--- BEECHFK.prj (project) ---

Proj Title=BEECHFK
Current Plan=p01
Default Exp/Contr=0,0
English Units
Geom File=g01
Flow File=f01
Plan File=p01
BEGIN DESCRIPTION:
END DESCRIPTION:
DSS Export Rating Curves= 0
DSS Export Rating Curve Sorted= 0
DSS Export Volume Flow Curves= 0
DXF OffsetX= 0
DXF OffsetY= 0
DXF ScaleX= 0
DXF ScaleY= 0

--- BEECHFK.p01 (plan) ---

Plan Title=Floodplain
Program Version=4.00
Geom File=g01
Flow File=f01
K Sum by GR=0
Std Step Tol=0.01
Critical Tol=0.01
Num of Std Step Trials=20
Max Error Tol=0.3
Flow Tol Ratio=0.001
Split Flow NTrial=30
Split Flow Tol=0.02
Split Flow Ratio=0.02
Log Output Level=0
Friction Slope Method=1
Unsteady Friction Slope Method=2
Unsteady Bridges Friction Slope Method=1
Global Log Level=0
CheckData=False
Run HTab=0
Run UNet=0
Run PostProcess=0
UNET Theta=0
UNET Theta Warmup=0
UNET ZTol=0
UNET ZSATol=0
UNET MxIter=0
UNET MaxInSteps=0
UNET DtIC=0
UNET DtMin=0
UNET MaxCRTS=0
UNET WFStab=0
UNET SFStab=0
UNET WFX=0
UNET SFX=0
UNET DSS MLevel=0
UNET DZMax Abort=0
UNET Convert EG Bridges=0
UNET Use Existing IB Tables=0
UNET Froude Limit=0
UNET Froude Power=0
Write IC File=0
Echo Input=False
Echo Output=False
Write Detailed=0

--- BEECHFK.f01 (steady flow) ---

Flow Title=NFF Regression Equation
Program Version=4.00
Number of Profiles= 1
Profile Names=P100yr
River Rch & RM=BEECHFK,Main            ,123497.2
     344
River Rch & RM=BEECHFK,Main            ,121955.6
     374
River Rch & RM=BEECHFK,Main            ,121713.6
     427
River Rch & RM=BEECHFK,Main            ,120753.5
     450
River Rch & RM=BEECHFK,Main            ,120507.5
     611
River Rch & RM=BEECHFK,Main            ,117519.8
     677
River Rch & RM=BEECHFK,Main            ,116912.5
     734
River Rch & RM=BEECHFK,Main            ,115112.9
     812
River Rch & RM=BEECHFK,Main            ,112119.1
     892
River Rch & RM=BEECHFK,Main            ,111742.9
    1153
River Rch & RM=BEECHFK,Main            ,108498.2
    1258
River Rch & RM=BEECHFK,Main            ,106422.9
    1392
River Rch & RM=BEECHFK,Main            ,102495
    1458
River Rch & RM=BEECHFK,Main            ,102181.1
    1694
River Rch & RM=BEECHFK,Main            ,100384.5
    1802
River Rch & RM=BEECHFK,Main            ,92583.9
    1972
River Rch & RM=BEECHFK,Main            ,92267.3
    2608
River Rch & RM=BEECHFK,Main            ,83140.2
    2852
River Rch & RM=BEECHFK,Main            ,74279.4
    3160
River Rch & RM=BEECHFK,Main            ,64408.5
    3458
River Rch & RM=BEECHFK,Main            ,63144.9
    4288
Boundary for River Rch & Prof#=BEECHFK,Main            , 1
Up Type= 0
Dn Type= 3
Dn Slope=0.00033
DSS Import GetInterval= 0
DSS Import GetPeak= 0
DSS Import FillOption= 0

--- BEECHFK.g01 (geometry) ---

Geom Title=USGS 10m DEM
Program Version=4.00

River Reach=BEECHFK         ,Main
Reach XY= 30
     1599235.167      428160.654     1599990.681       433328.67
     1598413.124      436822.244     1598431.962      444913.036
     1596063.065      447317.043     1594789.988       446693.42
     1592392.988      448533.128     1590530.139      453994.238
     1591801.686      455523.375     1590159.224      455446.854
     1589817.539      459921.419     1588219.196      462189.327
     1591159.621      465703.421     1590879.916       467428.72
     1592534.218       467893.85     1594715.082      471438.613
     1593418.876      477485.746     1590784.947      479295.006
     1590136.661      476805.234     1588016.017      474985.303
     1584766.399      477149.409     1584774.995      478445.244
     1578458.486      478743.461     1578674.759      480836.672
     1573758.417      479589.242     1572819.947      482422.028
     1568686.781      479929.163     1567460.299      476281.676
     1564787.606      477416.272     1562681.277      476713.478

Type RM Length L Ch R = 1 ,123497.2,786,782.9,780.9
XS GIS Cut Line= 3
     1598360.043      428514.348     1599241.697      428168.228
     1600039.558      427746.365
#Sta/Elev= 30
    10.1  947.39   191.4  931.71   221.7  927.88   251.9  921.08   312.4  915.33
   483.7  878.64   503.8   871.1     534  856.34   564.3  845.24   594.5  837.18
     655   825.7   675.1  824.17   725.5   823.8   932.2  809.79   947.2  808.65
   957.3  810.58   987.7  824.86  1089.1  865.78    1150  888.09  1210.8  908.41
  1241.2  917.59  1393.4  956.83  1494.8  988.93  1565.7 1016.23  1677.3 1064.27
  1687.4 1067.44  1707.7 1069.11  1748.3  1069.4  1778.7 1064.07  1849.7 1055.13
#Mann= 3 , 0 , 0
    10.1     .06       0   932.2    .045       0   957.3     .06       0
Bank Sta=932.2,957.3
XS Rating Curve= 0 ,0
Exp/Cntr=0.3,0.1

Type RM Length L Ch R = 1 ,122714.3,226.8,224.6,220.4
XS GIS Cut Line= 4
      1598928.07      429373.837     1599339.577      429071.648
     1599845.768      428665.074     1600292.711      428154.662
#Sta/Elev= 30
      10 1039.08    70.1 1014.51   110.1  1002.1   210.2  966.15   270.3  947.47
   340.4  932.97   390.4  931.28   460.5  909.51   500.5  901.45   601.8  856.88
   672.9  819.74   713.4  804.61   743.9  800.08   794.6  801.53     881  800.21
     896  799.46     911  800.28   926.5  805.77  1068.5  881.89  1098.9  895.89
  1311.7  956.93  1382.6  980.17  1423.1  986.16  1483.8  991.21  1514.2  988.17
    1575  974.77  1605.3  970.92  1757.2  971.56  1777.5  974.06  1838.2  987.75
#Mann= 3 , 0 , 0
      10     .06       0     881    .045       0     911     .06       0
#XS Ineff= 2 , 0
          870.96  818.47
Permanent Ineff=
       F       F
Bank Sta=881,911
XS Rating Curve= 0 ,0
Exp/Cntr=0.3,0.1

Type RM Length L Ch R = 1 ,122489.7,36.7,37.8,38.6
XS GIS Cut Line= 4
      1599038.13      429436.073     1599676.407      429177.377
     1599939.208      428765.817     1600652.176      428369.767
#Sta/Elev= 30
    10.1 1021.41   141.8  977.91   232.9  952.07   435.5  913.16   536.8  888.94
   638.1  849.75   768.4  805.18   798.3  801.15   932.8  797.76   947.8  797.14
   957.8  798.46   997.6  820.49  1027.5  832.96  1147.1  896.93    1177  906.08
  1348.2  945.97  1368.3  946.78  1398.5  942.64  1539.5  914.48  1589.8  908.55
  1620.1  907.93  1650.3  910.29  1690.5  921.47  1720.7  924.69  1740.9  924.48
  1801.3  916.47  1831.5  918.76  1881.8  932.85  1952.3  960.72  1992.6  969.88
#Mann= 3 , 0 , 0
    10.1     .06       0   932.8    .045       0   957.8     .06       0
Bank Sta=932.8,957.8
XS Rating Curve= 0 ,0
Exp/Cntr=0.3,0.1

Type RM Length L Ch R = 1 ,122451.9,52.9,52.6,55.2
XS GIS Cut Line= 4
     1599047.801      429455.415     1599678.825      429196.719
     1600011.991      428764.074     1600701.661       428593.38
#Sta/Elev= 30
      10 1018.73    20.1 1018.03   130.4  981.96   210.6  960.11   300.9   941.1
   451.3  914.98   531.6  895.43     682  839.43   742.7  814.04     773  804.76
   803.3  800.36     940   797.7  955.09  797.08  962.35  799.05  1035.9  829.33
  1126.9  874.86  1177.5  895.38  1228.1  912.64  1339.7  936.41  1390.4  934.73
  1441.2  926.02  1583.3  875.64  1603.6   870.8  1644.2  879.96  1664.5  880.08
  1694.9  877.59  1745.7  866.26    1766  864.63  1816.7  884.85  1938.5  896.55
#Mann= 3 , 0 , 0
      10     .06       0     940    .045       0  962.35     .06       0
Bank Sta=940,962.35
XS Rating Curve= 0 ,0
Exp/Cntr=0.3,0.1

Type RM Length L Ch R = 1 ,122399.3,66.5,67.2,68
XS GIS Cut Line= 4
     1599067.143      429469.921      1599705.42      429208.808
     1600006.175      428875.626     1600716.735        428682.6
#Sta/Elev= 30
    10.1 1015.71    30.4 1011.64   131.8  979.72   202.8  962.21   294.1  943.68
   436.1  920.73   517.2  901.36   557.8   887.6   638.9  854.43   789.4  801.54
   849.2  798.76   953.9  797.74   968.9  796.94   978.9   797.9   988.9  801.15
  1018.8  817.55  1138.5  867.96  1289.8  909.68  1309.9  913.43  1350.3  913.62
  1461.2  892.08  1491.5  879.84  1541.9  846.31  1562.1  840.62  1582.3  841.61
  1602.4  845.87  1673.1  849.29  1733.6  847.97  1794.1  862.39  1874.8  873.58
#Mann= 3 , 0 , 0
    10.1     .06       0   953.9    .045       0   978.9     .06       0
Bank Sta=953.9,978.9
XS Rating Curve= 0 ,0
Exp/Cntr=0.3,0.1

Type RM Length L Ch R = 1 ,122332.1,128.3,132.1,133.3
XS GIS Cut Line= 5
     1599074.396      429486.845     1599719.926      429242.656
     1600084.504      428903.601     1600327.885      428892.411
     1600764.293      428917.588
#Sta/Elev= 30
    10.1 1011.22    30.4 1012.11   131.9  982.01   223.3  961.29   294.3  947.95
   426.3  929.41   537.9  903.07   639.4   862.1   781.6  808.96   812.1  799.77
   862.9  797.57  1000.3  797.42  1015.3  796.36  1020.3  797.66  1025.5     799
    1056  817.62    1188  870.41  1289.6  889.74  1330.2  881.64  1401.2  854.36
  1451.6  841.46  1491.3  828.52    1531  822.89  1560.8  821.32  1640.3  822.72
    1690  813.12  1769.5  813.22  1789.3   815.3  1819.1  823.78  1868.8  829.63
#Mann= 3 , 0 , 0
    10.1     .06       0  1000.3    .045       0  1020.3     .06       0
Bank Sta=1000.3,1020.3
XS Rating Curve= 0 ,0
Exp/Cntr=0.3,0.1

Type RM Length L Ch R = 1 ,122200  ,241.5,244.4,246.9
XS GIS Cut Line= 5
      1599066.22       429505.06     1599654.869      429320.138
     1599831.308      429253.041      1600166.79      429019.446
      1600778.28       428981.93
#Sta/Elev= 30
    10.1 1001.94    40.5 1011.41    50.6 1011.64   151.7  983.69   202.3  972.41
   293.3  955.52   414.7  940.21   475.4  925.74   566.4  907.68   586.7  901.83
   626.9  883.91   666.7  870.34   746.2  839.39   825.7  810.94   865.6  799.34
   935.4  796.24  1079.9   795.6  1094.9  794.99  1104.9  795.67  1144.8  812.99
  1214.6  834.12  1244.7  832.01    1315  814.48  1345.1  809.81    1546  808.17
  1586.2  812.18  1656.5  829.57  1736.8  843.43    1787  849.81  1827.2  851.83
#Mann= 3 , 0 , 0
    10.1     .06       0  1079.9    .045       0  1104.9     .06       0
#XS Ineff= 2 , 0
          954.55  802.22
Permanent Ineff=
       F       F
Bank Sta=1079.9,1104.9
XS Rating Curve= 0 ,0
Exp/Cntr=0.3,0.1

Type RM Length L Ch R = 1 ,121955.6,240.6,242.1,243.5
XS GIS Cut Line= 4
     1599100.439      429600.175     1599871.069      429260.496
     1600194.126       429198.37     1600964.793      429426.608
#Sta/Elev= 30
    10.1  977.51    81.2 1007.93    91.3 1010.55   101.5 1010.55   202.9  984.91
   253.7  974.05   355.1   956.1   578.4  909.39   598.7  903.25   629.1  890.85
   659.5  881.72     761  839.37   842.2  810.33     892  796.57   951.8   794.7
   976.7  791.97   991.7     791  1006.7  791.86  1031.6  794.01  1081.4  793.37
  1161.2   796.8  1251.5  809.01  1321.9  829.04  1482.6  898.68  1593.1  928.82
  1713.7  957.41  1733.8  960.49  1824.2  966.68  1884.5  973.93  1974.9  974.49
#Mann= 3 , 0 , 0
    10.1     .06       0   976.7    .045       0  1006.7     .06       0
#XS Ineff= 2 , 0
                          1024.1          814.22
Permanent Ineff=
       F       F
Bank Sta=976.7,1006.7
XS Rating Curve= 0 ,0
Exp/Cntr=0.3,0.1

Type RM Length L Ch R = 1 ,121713.6,489.1,493.7,498.3
XS GIS Cut Line= 4
     1599117.687      429632.571     1599778.009      429510.555
     1600402.444      429417.249       1600989.8      429464.188
#Sta/Elev= 30
      10  974.18   100.2 1007.08   110.2 1009.97   120.3 1011.27   210.5  999.03
   310.7  980.83     451  961.81   521.2  949.72   581.3   935.7   681.5  906.62
   691.5  902.86   791.8  854.54   851.9  824.11     882  811.59   937.1  791.23
   942.1  790.08   952.1  790.02   967.1  791.56  1112.5  797.45  1122.5  798.49
  1162.6   808.6  1182.6  816.61  1353.7  897.06    1374  905.67    1567  955.37
  1648.3  973.58  1688.9   984.1  1709.2  986.66  1749.9  989.38  1892.1  987.16
#Mann= 3 , 0 , 0
       0     .06       0   937.1    .045       0   967.1     .06       0
Bank Sta=937.1,967.1
XS Rating Curve= 0 ,0
Exp/Cntr=0.3,0.1

Type RM Length L Ch R = 1 ,121219.9,263.2,262.2,261.2
XS GIS Cut Line= 3
     1599314.639      429712.976     1600029.205       429947.09
     1600886.493      430222.573
#Sta/Elev= 30
    10.2  984.59   132.1 1013.95   142.3 1014.56   162.6 1011.44   182.9 1004.74
   233.7  981.35     254  974.05     376  949.85   477.6  921.77   548.7  899.44
   579.2  885.38   650.3  846.42   711.3  820.91   731.6  806.76   751.9  789.97
   757.2   787.8   762.1   785.8   772.2  785.66   787.2  788.29   984.6  799.42
  1055.5  819.12  1116.2  830.14  1207.2  851.12  1298.3  877.88  1328.6   885.2
  1369.1  892.48  1419.7  888.85  1439.9  889.15  1581.6  932.16  1652.4   939.4
#Mann= 3 , 0 , 0
       0      .1       0   757.2    .045       0   787.2      .1       0
Bank Sta=757.2,787.2
XS Rating Curve= 0 ,0
Exp/Cntr=0.3,0.1

Type RM Length L Ch R = 1 ,120957.7,201.8,204.2,206.6
XS GIS Cut Line= 4
     1599118.251      430029.598     1599828.847      430164.097
     1600054.104      430212.975      1600860.33      430282.532
#Sta/Elev= 30
      10  871.28    60.3  876.46   100.4  891.69   130.6  898.26   251.1  896.32
   532.4  884.08   632.8  864.86   723.2  827.67   793.4  790.99   813.4  784.83
   828.5  783.05   843.5   782.8   858.5  782.91   893.6  785.08  1024.5   800.8
  1075.1  818.36  1115.6  824.03  1166.1  822.16  1257.2  813.21  1338.1  810.66
  1348.2  812.87  1378.6  826.48    1419  838.61  1439.2   841.3  1469.6  840.66
  1510.1  861.75  1530.3  869.82  1621.3  893.41  1732.6  925.75  1762.9  931.62
#Mann= 3 , 0 , 0
       0      .1       0   828.5    .045       0   858.5      .1       0
Bank Sta=828.5,858.5
XS Rating Curve= 0 ,0
Exp/Cntr=0.3,0.1

Type RM Length L Ch R = 1 ,120753.5,247.9,246.1,244.2
XS GIS Cut Line= 4
     1599065.505      430065.064     1599752.916      430290.648
     1600034.944      430428.046      1600812.21      430662.913
#Sta/Elev= 30
      10  860.58    50.2  856.87   150.7  869.31   180.9  870.52   321.5  863.44
   442.1     853   492.4  850.65   522.5  846.95   582.8  833.61   653.1  821.65
   703.4  807.07   753.8  789.08   784.2  787.29   895.5  786.97     921  784.26
     936  782.79   946.1  785.05   976.5  802.39  1189.4  884.63    1230  897.72
  1290.9  908.76    1362  915.48  1412.7  912.89  1473.6  906.61  1514.2  905.99
  1554.8  907.93  1615.7  916.19  1646.2  918.03  1717.2  918.72  1849.2  914.78
#Mann= 3 , 0 , 0
      10     .06       0     921    .045       0   946.1     .06       0
Bank Sta=921,946.1
XS Rating Curve= 0 ,0
Exp/Cntr=0.3,0.1

Type RM Length L Ch R = 1 ,120507.5,414.3,414.8,415.3
XS GIS Cut Line= 3
     1598926.778      430566.397     1599547.478      430520.263
     1600747.131       430845.08
#Sta/Elev= 30
      10  871.13    30.1  865.08    90.4  842.59   140.5  818.77   180.7  806.18
   200.8  801.88   220.9  801.39   321.2  806.46   431.7  804.21   461.8  801.45
     522  792.82   552.1  791.74   592.3  787.23   672.9  783.87   733.6  789.74
   784.1  782.22   885.1  781.01   910.5  779.18   925.5  778.57   935.6  780.92
     966  795.72    1067  832.31  1178.2  885.26  1198.4  893.41  1289.3  910.11
  1440.9  950.07  1461.1  952.25  1632.9  958.24  1794.5  957.12  1865.3  959.59
#Mann= 3 , 0 , 0
      10     .06       0   910.5    .045       0   935.6     .06       0
#XS Ineff= 2 , 0
          847.06  800.86
Permanent Ineff=
       F       F
Bank Sta=910.5,935.6
XS Rating Curve= 0 ,0
Exp/Cntr=0.3,0.1

Type RM Length L Ch R = 1 ,120092.7,302.4,303.4,303
XS GIS Cut Line= 4
     1598895.438      430692.663     1599401.057      430870.718
     1599989.316       431062.33     1600635.283      431263.298
#Sta/Elev= 30
    10.1  871.42    60.7  852.97   151.7  813.69   161.8  812.13   202.3  811.75
   232.6  814.87   273.1  824.97   303.4  836.82   374.2  868.57   424.8  886.69
   475.4  892.72   515.8  893.94   546.2  887.98   617.2  862.84   698.3  830.67
   759.2  802.47   799.8  784.94   809.9  782.11   977.5  778.19   992.5  777.29
  1002.6  779.73    1033  794.35  1124.3  833.82  1195.1   870.7  1306.2  897.18
  1528.3  959.52  1629.3  995.73  1790.9 1063.68    1811 1070.12  1831.2 1073.47
#Mann= 3 , 0 , 0
    10.1     .06       0   977.5    .045       0  1002.6     .06       0
Bank Sta=977.5,1002.6
XS Rating Curve= 0 ,0
Exp/Cntr=0.3,0.1

Type RM Length L Ch R = 1 ,119789.2,110.8,115.1,120.9
XS GIS Cut Line= 4
     1598939.905      430812.225     1599622.496      431159.103
     1599923.755      431267.247     1600533.385      431441.397
#Sta/Elev= 30
    10.1  845.78    50.4  826.78    80.6  816.48    90.7  815.73   120.9  820.57
   161.2  829.95   221.6  849.22   352.6  900.61   382.8  908.76     403  910.39
   483.6  894.37   564.2  871.17   604.5  854.12   755.6  780.75   830.7   776.2
   845.6  776.08   860.7  776.23   915.7  781.32   985.7  806.22  1075.8  833.92
    1126  852.77  1156.2  867.12  1216.6  882.91  1266.9  902.33  1417.9  951.94
  1518.5  988.31  1558.8  999.75    1599 1016.38  1679.5 1056.35  1719.8  1067.9
#Mann= 3 , 0 , 0
    10.1     .06       0   830.7    .045       0   860.7     .06       0
Bank Sta=830.7,860.7
XS Rating Curve= 0 ,0
Exp/Cntr=0.3,0.1

Type RM Length L Ch R = 1 ,119674.1,162.3,154.7,147.1
XS GIS Cut Line= 4
     1598944.658      430931.314     1599560.868      431146.106
     1599759.461      431391.427     1600503.043      431574.917
#Sta/Elev= 30
      10  827.18    70.3   829.6   120.5   840.6   160.6  852.31     261  887.96
   341.3  909.89   361.4  912.85   381.5  909.59   451.8  893.63     512  875.92
   562.2  853.91   652.6  807.35   731.5  779.07   751.2  776.88   790.7  778.08
     825  777.37  840.15  775.95     855   777.8   928.7  784.71   968.2  790.37
  1048.8  814.91  1099.2  831.93  1210.1  875.59  1371.3  921.88  1472.1  953.91
  1532.5  976.39    1593 1004.54  1643.4 1022.61  1673.6 1029.01  1734.1 1032.61
#Mann= 3 , 0 , 0
      10     .06       0     825    .045       0     855     .06       0
Bank Sta=825,855
XS Rating Curve= 0 ,0
Exp/Cntr=0.3,0.1

Type RM Length L Ch R = 1 ,119519.4,426.4,423.3,419.1
XS GIS Cut Line= 4
      1598751.68      431107.663     1599455.129      431375.391
     1599823.335      431462.936     1600512.546      431648.372
#Sta/Elev= 30
      10   865.1    30.1  863.87    40.1  865.79    80.3  884.71   100.4  889.74
   200.7  894.51   311.1  911.03   431.5  923.24   471.7  932.74   491.7  933.22
   531.9  928.16     552  922.98   652.3  886.29   762.6  834.54   842.3  788.54
   877.1   773.4   892.1  771.72   907.1  771.83  1041.5  784.16  1111.2  800.48
  1231.7   839.7  1271.9  856.23  1312.1  877.16  1543.3   938.3  1613.7  959.24
  1633.8  966.26    1684  991.86  1714.2 1002.16  1784.6 1010.61  1844.9 1007.54
#Mann= 3 , 0 , 0
       0     .06       0   877.1    .045       0   907.1     .06       0
Bank Sta=877.1,907.1
XS Rating Curve= 0 ,0
Exp/Cntr=0.3,0.1

Type RM Length L Ch R = 1 ,119096.1,799.5,798.5,798.5
XS GIS Cut Line= 3
     1598745.796      431875.311     1599649.738      431813.636
     1600612.144      431646.939
#Sta/Elev= 30
    10.1 1020.72    90.6  990.07   261.7  929.77   312.1  917.93   382.6  910.22
     453  898.98   563.8  873.26   674.5   842.7   724.8  826.91     745  818.84
   825.5  780.66   845.6  775.68     891  770.61     906  769.64     921  770.25
    1047   780.2  1087.3  787.38  1107.4  793.71  1198.1  829.82  1248.4  852.31
  1288.7  873.21  1308.8  880.43  1490.1  923.82  1580.7  947.54  1600.8  954.36
  1641.1  973.45  1711.6  992.68  1761.9  996.93  1802.2 1003.22  1882.8 1022.27
#Mann= 3 , 0 , 0
       0     .06       0     891    .045       0     921     .06       0
Bank Sta=891,921
XS Rating Curve= 0 ,0
Exp/Cntr=0.3,0.1

Type RM Length L Ch R = 1 ,118297.6,783.8,777.8,771.8
XS GIS Cut Line= 3
     1598781.653      432549.187     1599364.881       432368.62
     1600637.019      432405.976
#Sta/Elev= 30
      10  910.09   110.1   908.4   190.2  908.64   250.2  910.49   340.3  916.38
   430.4  920.19   490.4  920.95   510.5  918.92   530.5  914.79   610.5  889.79
   671.1  873.91   701.4   863.5   762.1  836.69   898.6  767.64   903.5  765.89
   913.6  764.81   928.6  766.59   943.9  768.65  1034.8  771.27    1055  776.21
  1196.4  848.34  1236.8  866.47  1307.5   895.6  1398.4  930.54  1590.3  999.82
  1751.9 1053.65  1802.4 1068.15  1822.6 1070.88  1842.8  1069.8  1883.2 1064.63
#Mann= 3 , 0 , 0
       0     .06       0   898.6    .045       0   928.6     .06       0
Bank Sta=898.6,928.6
XS Rating Curve= 0 ,0
Exp/Cntr=0.3,0.1

Type RM Length L Ch R = 1 ,117519.8,598.1,607.3,616.9
XS GIS Cut Line= 4
     1598850.756      433099.328     1599679.046      433175.451
     1600216.818      432860.013      1600659.18      432616.129
#Sta/Elev= 30
    10.1  865.11   101.4  867.06   152.2  863.17   243.4  866.75   324.6  862.24
   446.3  869.58   547.8  872.39   578.2   868.4   628.9  858.57   740.5  833.25
   770.9  821.94   811.5  802.28   892.1  771.52   902.2  769.01    1043  764.38
  1068.2  761.84  1083.2  761.14  1098.2  763.71  1123.4  769.18  1133.5  773.13
  1254.1  829.74  1334.6  863.78    1415  889.26  1455.2   900.1  1546.2  915.59
  1616.9  923.25  1677.5  934.49  1738.1  948.05  1859.3  970.52  1960.4  983.26
#Mann= 3 , 0 , 0
       0     .06       0  1068.2    .045       0  1098.2     .06       0
Bank Sta=1068.2,1098.2
XS Rating Curve= 0 ,0
Exp/Cntr=0.3,0.1

Type RM Length L Ch R = 1 ,116912.5,782.5,781.6,780.3
XS GIS Cut Line= 3
     1598921.434      433163.304     1599756.548      433487.851
     1600660.123      433891.293
#Sta/Elev= 30
    10.1  884.23    80.5  888.03   171.1     896   382.5  910.98   402.7  910.34
   543.6  873.72   674.5  843.44   734.9  827.74   785.2  806.95   865.8  771.39
   885.9  761.21   891.1  760.04   906.1  758.82   921.1  759.86  1077.7  769.05
  1097.9  771.79    1108  775.81  1138.3  791.05  1148.4  794.09  1198.9  801.65
    1209  805.03  1269.6  839.12  1289.8  847.85  1380.6   869.3    1421  881.42
  1481.6  902.25  1612.9  951.25  1734.1  980.77  1824.9  994.22  1885.5 1016.39
#Mann= 3 , 0 , 0
       0     .06       0   891.1    .045       0   921.1     .06       0
Bank Sta=891.1,921.1
XS Rating Curve= 0 ,0
Exp/Cntr=0.3,0.1

Type RM Length L Ch R = 1 ,116130.9,1015.8,1018,1020.4
XS GIS Cut Line= 3
     1598697.381      433926.119       1599422.3      434141.441
     1600412.783      434435.715
#Sta/Elev= 30
    10.1 1023.67   100.8  982.75   131.1  970.47   292.4  911.83   403.3  876.41
   433.6  868.35     484  859.57   504.1  854.63   544.5  840.69   695.7  794.18
     817  760.86   837.3  758.79   908.2  757.61   943.8  755.58   958.8  753.93
   973.8  756.02  1070.3  800.05  1120.9  826.02    1131  830.06  1171.6  836.44
  1252.6  854.59  1293.1  865.18  1333.6  881.18  1414.7  908.54  1434.9   914.4
  1465.3  920.48  1485.6  926.58  1566.6  955.35    1597  967.78  1789.5 1033.59
#Mann= 3 , 0 , 0
       0     .06       0   943.8    .045       0   973.8     .06       0
Bank Sta=943.8,973.8
XS Rating Curve= 0 ,0
Exp/Cntr=0.3,0.1

Type RM Length L Ch R = 1 ,115112.9,249.2,248.6,247.6
XS GIS Cut Line= 3
     1598341.085      434640.191     1599151.643      435031.247
     1599927.294      435487.126
#Sta/Elev= 30
    10.1  927.93   141.6  907.58   232.6  889.72   283.1  883.61   353.9  880.32
   434.8  888.14     455     889   475.3  888.24   495.5  884.81   616.8  852.62
   657.3  838.03   728.1  816.84   839.3  778.02   869.6  763.12   889.8  751.75
     900  747.82   910.1  746.44   930.3  746.87  1263.9  759.65  1334.6  776.52
  1395.3  786.29    1456  793.22  1496.4  796.46  1546.9  803.38  1617.7  815.43
  1637.9  817.64  1688.5  812.41  1718.8  807.64  1749.1  800.58  1799.7  784.81
#Mann= 3 , 0 , 0
    10.1      .1       0     900    .045       0   930.3     .06       0
Bank Sta=900,930.3
XS Rating Curve= 0 ,0
Exp/Cntr=0.3,0.1

Type RM Length L Ch R = 1 ,114864.3,419.9,403.2,386.6
XS GIS Cut Line= 4
     1598227.735      434949.509     1598891.686      435148.694
     1599173.074      435281.485     1599925.551      435657.723
#Sta/Elev= 30
       0  841.89    80.4  838.89   140.6  822.12   160.7  818.99   180.8  819.02
     221  822.44   341.6  800.71   381.8  808.36   482.2   817.9   522.4  820.21
   542.5  818.79   602.8  806.36   673.1  788.21   693.2  781.51   753.4  752.79
   781.1  745.14   793.6  744.42   806.1   744.7  1065.1  750.12  1146.2   756.1
  1166.5  762.44  1318.6   821.9  1338.8  827.69  1389.5  839.49    1430  846.68
    1572  861.33  1632.8   861.9    1724  856.41  1784.8  844.27  1845.6  824.95
#Mann= 3 , 0 , 0
       0      .1       0   781.1    .045       0   806.1     .06       0
Bank Sta=781.1,806.1
XS Rating Curve= 0 ,0
Exp/Cntr=0.3,0.1

Type RM Length L Ch R = 1 ,114461.1,954.7,965.1,975.3
XS GIS Cut Line= 4
     1598108.833      435218.053     1598814.961      435624.192
     1599149.867      435417.081     1599850.311      435998.958
#Sta/Elev= 30
    10.1  775.09    30.2   776.8    80.5  790.45   211.2  808.92   261.5  810.88
   321.8  804.78     352  804.84   492.8  825.51   593.3  829.31   623.5  823.42
   693.9  795.42   834.8  750.43  1097.3  745.88  1122.7  743.57  1137.7  742.88
  1152.7  745.63  1178.1  749.08  1238.7  750.02    1259  753.71  1390.5  816.15
  1410.7  823.17  1441.1   829.2  1481.5  833.09    1522  842.03  1663.7   887.3
  1744.6  906.93  1805.3  915.02  1926.7  913.53    2038  908.81    2119  898.15
#Mann= 3 , 0 , 0
       0     .06       0  1122.7    .045       0  1152.7     .06       0
Bank Sta=1122.7,1152.7
XS Rating Curve= 0 ,0
Exp/Cntr=0.3,0.1

Type RM Length L Ch R = 1 ,113496.1,875.6,871.8,868.1
XS GIS Cut Line= 3
     1597949.697      435762.486     1598716.355      436249.472
      1599479.72      436718.133
#Sta/Elev= 30
    10.1  999.79    70.6 1000.83   131.2 1006.37   171.6 1005.06   201.8  998.93
     222  991.44   252.3  974.51   292.7  956.43   383.5  921.45   484.4  886.87
   696.3  824.16   736.7   802.3   797.2  761.55   827.5  746.74   857.8  739.59
   893.3  738.15   908.3  737.45   923.3  738.23   998.8  743.05    1019  746.85
  1099.5   782.2    1180   810.5  1220.3  827.09  1300.8  849.53  1471.9  888.89
  1522.2  902.72    1643   961.4  1733.5 1009.23  1773.8 1034.61    1804 1046.75
#Mann= 3 , 0 , 0
       0     .06       0   893.3    .045       0   923.3     .06       0
Bank Sta=893.3,923.3
XS Rating Curve= 0 ,0
Exp/Cntr=0.3,0.1

Type RM Length L Ch R = 1 ,112624.3,504.2,505.2,505.7
XS GIS Cut Line= 3
     1597606.414      436883.213     1598460.732      437012.433
     1599336.171       437170.31
#Sta/Elev= 30
      10  964.95    40.2  961.29   100.5  949.77   261.2  910.53   291.4  905.42
   351.6  898.43   442.1  880.96   492.3  869.33   552.6  845.88     653  810.81
   683.2  794.98   763.6  748.85   793.7  740.69   859.1  732.97   874.1  731.28
   889.1   732.5   985.3  738.64   995.4  742.21  1025.8  757.84  1096.5  778.01
  1207.7  824.63  1258.3  843.65  1318.9  847.62  1369.5  858.58  1470.6  875.53
  1561.5  887.67  1591.9  893.77  1652.5  912.43  1723.3  944.53  1753.6     956
#Mann= 3 , 0 , 0
       0     .06       0   859.1    .045       0   889.1     .06       0
Bank Sta=859.1,889.1
XS Rating Curve= 0 ,0
Exp/Cntr=0.3,0.1

Type RM Length L Ch R = 1 ,112119.1,113.5,115.8,118.4
XS GIS Cut Line= 4
     1597575.357      437219.231      1598416.36      437465.842
     1598615.546      437497.458     1599301.628      437478.488
#Sta/Elev= 30
    10.1  967.18   110.8  922.55   161.2  904.32   211.5  891.11   292.1  877.21
   322.4  869.96   382.8  852.51   493.6  815.82   564.1  798.84   604.4   786.2
   634.6   781.5   695.1  777.25   856.3  745.01   886.5  736.74   952.2  730.77
   967.2   728.9   982.2  730.29  1017.6   741.9  1057.9  761.84  1108.4  807.04
  1128.6  820.81  1138.7  825.07  1239.6  858.65  1330.4  883.55  1370.8  897.44
  1431.4  923.57  1582.8  997.06  1643.3 1018.79  1683.7 1030.58  1764.4 1041.43
#Mann= 3 , 0 , 0
       0     .06       0   952.2    .045       0   982.2     .06       0
Bank Sta=952.2,982.2
XS Rating Curve= 0 ,0
Exp/Cntr=0.3,0.1

Type RM Length L Ch R = 1 ,112003.3,266.3,260.4,254.4
XS GIS Cut Line= 4
      1597562.71      437282.465     1598350.514      437519.013
     1598595.125       437655.48     1599472.358      437712.452
#Sta/Elev= 30
    10.2  942.56   121.9  908.41   172.6  895.27   253.9  878.44   528.1  804.04
   578.8   795.5   710.8  778.89   731.2  773.01   761.6  759.38   781.9  752.75
   842.6  745.14   872.6  735.25   947.6  730.14   962.6  728.41   977.6  730.54
  1052.6  756.35  1062.6  762.22  1102.7  798.72  1122.9  813.76  1213.8  852.81
  1314.8  881.77  1415.9  913.73  1486.6  939.02  1537.1  961.55  1638.2  997.07
  1698.8 1010.45  1769.5 1008.05  1840.3 1015.28  1900.9 1032.18  1981.7    1047
#Mann= 3 , 0 , 0
       0     .06       0   947.6    .045       0   977.6     .06       0
Bank Sta=947.6,977.6
XS Rating Curve= 0 ,0
Exp/Cntr=0.3,0.1

Type RM Length L Ch R = 1 ,111742.9,74.1,72.9,71.6
XS GIS Cut Line= 4
     1597468.475       438227.18     1598225.521      437818.616
      1598602.85      437835.721     1599429.005      437763.266
#Sta/Elev= 30
       0  797.75    10.1  797.75   141.7   778.6   192.3  773.53   263.1  767.98
   374.5  763.91   445.3  759.08   495.9  747.19   526.3  742.61   759.1  734.51
   979.5   731.6  1006.8  727.49  1019.3  726.19  1031.8  729.75  1049.1  738.49
  1098.8  759.47  1128.6  765.29    1228  809.44  1359.3  852.98  1440.2  876.36
  1470.6  884.44  1500.9   890.3  1541.4  892.47  1571.7  896.81  1672.9   922.6
  1824.6  954.94  1945.9  971.81  1976.3  980.84  1996.5  989.05  2067.3 1024.89
#Mann= 3 , 0 , 0
       0     .06       0  1006.8    .045       0  1031.8     .06       0
Bank Sta=1006.8,1031.8
XS Rating Curve= 0 ,0
Exp/Cntr=0.3,0.1

Type RM Length L Ch R = 1 ,111670  ,474.5,468.8,463
XS GIS Cut Line= 4
     1597505.931      438246.922     1598080.124      437923.938
     1598769.156      437866.519     1599508.747      437756.183
#Sta/Elev= 30
    10.1  811.52    81.1  804.75   263.5  772.31   425.7  762.36     527  743.41
   919.3  731.23   944.4  728.81   959.4  726.13   969.4  726.81   974.4  729.23
   979.5   731.7   999.5  747.86  1009.5   753.3  1029.6   758.8  1069.6  761.27
  1089.7  764.92  1119.7  776.21  1199.9  813.84  1320.2  855.22  1431.1  884.33
  1451.3  886.16  1491.7  884.04    1522  885.46    1613  910.62  1683.7  927.22
  1885.8  963.32  1936.3  980.15  2017.2 1022.75  2037.4 1031.53    2098 1043.02
#Mann= 3 , 0 , 0
       0     .06       0   944.4    .045       0   974.4     .06       0
Bank Sta=944.4,974.4
XS Rating Curve= 0 ,0
Exp/Cntr=0.3,0.1

Type RM Length L Ch R = 1 ,111201.3,102.5,105.2,109.6
XS GIS Cut Line= 4
     1597716.337      438645.004     1598508.579      438342.087
     1598733.825      438167.328     1599514.416      438008.103
#Sta/Elev= 30
    10.1  959.59    50.5  949.81    80.8  939.94   191.8  916.84   252.4  890.99
   262.5  888.36   343.3  881.39   504.9  832.43   595.7  808.33   696.7  767.11
   747.2  751.44   838.1  736.44   970.8  724.97   985.8  723.35  1000.8  724.77
  1044.8  731.17  1133.3  760.76  1234.1  778.97  1294.6  802.72  1435.8  835.66
  1536.6  848.74  1607.2  860.81  1647.6  864.67  1687.9  874.07  1748.4  903.79
  1829.1  954.31  1859.3  970.74  1899.7  986.73  1919.8  990.17  1929.9  988.29
#Mann= 3 , 0 , 0
       0     .06       0   970.8    .045       0  1000.8     .06       0
Bank Sta=970.8,1000.8
XS Rating Curve= 0 ,0
Exp/Cntr=0.3,0.1

Type RM Length L Ch R = 1 ,111096.1,849.9,853.1,854.5
XS GIS Cut Line= 3
     1597746.155      438727.755     1598671.357      438342.996
     1599542.914      438145.056
#Sta/Elev= 30
    10.1  988.76   111.3  935.75   172.1  911.72   232.8  891.94   263.2  884.01
   313.8   881.6   344.1   877.6   384.6  868.94   455.5  849.99   576.9  816.29
   738.9  755.64   819.8  739.75   890.7  730.17     921  728.65   971.7  731.29
     987  727.76    1002  723.33    1017  725.37    1063  734.81  1245.8  762.45
  1377.8  790.96  1448.9  808.41  1489.5  815.65  1672.3  841.58  1692.6  847.77
  1804.4  903.49  1824.7  910.84  1834.8   911.4  1865.3  905.04  1895.8   906.5
#Mann= 3 , 0 , 0
       0     .06       0     987    .045       0    1017     .06       0
Bank Sta=987,1017
XS Rating Curve= 0 ,0
Exp/Cntr=0.3,0.1

Type RM Length L Ch R = 1 ,110243  ,898.5,898.7,898.8
XS GIS Cut Line= 3
     1597800.205      439187.163     1598919.881      439101.034
      1599616.09       439057.97
#Sta/Elev= 30
    10.1 1032.36    50.6 1014.68    91.1 1000.95   121.4  979.89   151.8  963.02
   232.7  913.12     263  897.66   293.4  885.58   414.8  847.74   566.6  812.38
     688  764.61   758.8  754.57     779  749.49   855.1  717.62   870.1  715.35
   885.1  717.77   961.1  728.32   991.5  745.01  1001.6  748.43  1112.9   764.4
  1234.2  808.59    1305  827.79  1385.8  846.52  1426.3  865.32    1497  885.71
  1618.3  939.04  1658.8  959.08  1699.2  981.98    1770 1029.74  1820.5 1044.33
#Mann= 3 , 0 , 0
       0     .06       0   855.1    .045       0   885.1     .06       0
Bank Sta=855.1,885.1
XS Rating Curve= 0 ,0
Exp/Cntr=0.3,0.1

Type RM Length L Ch R = 1 ,109344.3,437.9,442,446.1
XS GIS Cut Line= 3
     1597893.511      440048.453     1598814.709      440000.556
     1599725.614       439972.71
#Sta/Elev= 30
    10.1  920.25   121.6  913.83   192.6  906.84   233.1  901.71   304.1  888.91
   354.8  891.27   405.5  899.84   435.9  897.54   456.2  893.55   537.2  869.72
   658.9  837.66   699.4  824.41   760.3  801.05   790.7  787.21   871.8  734.77
   897.3  716.63   902.2  713.82   912.3  712.39   927.3  714.86  1165.5  731.95
  1185.7  737.81  1266.7  773.37  1307.2  789.07  1327.5   795.8    1368  805.48
  1408.5  809.54  1489.5  820.82  1661.6  831.28  1742.6  844.46  1833.8  854.79
#Mann= 3 , 0 , 0
       0     .06       0   897.3    .045       0   927.3     .06       0
Bank Sta=897.3,927.3
XS Rating Curve= 0 ,0
Exp/Cntr=0.3,0.1

Type RM Length L Ch R = 1 ,108902.3,272.3,272.8,273.3
XS GIS Cut Line= 4
     1597836.007      440536.747      1598589.72      440342.727
      1599034.72      440507.808     1599700.248      440690.802
#Sta/Elev= 30
    10.1  767.79    50.5  766.46   232.5  741.58   242.6  742.74   272.9  751.54
   293.1  754.89   495.3  775.93   576.1  791.24   636.8  800.08   687.3  804.64
   768.2  804.75   788.4  799.81   818.7  787.01   859.1  765.25   929.8  722.85
   939.9  718.84  1015.7  713.05  1030.7  711.35  1045.7  712.57  1131.7  723.97
  1242.8  749.27  1344.3  783.85  1496.5  828.36  1557.4  843.64  1638.6  858.06
  1658.9  862.95  1750.3  898.17  1790.9  909.04  1831.5  914.76  1943.1  920.34
#Mann= 3 , 0 , 0
       0     .08       0  1015.7    .045       0  1045.7     .08       0
Bank Sta=1015.7,1045.7
XS Rating Curve= 0 ,0
Exp/Cntr=0.3,0.1

Type RM Length L Ch R = 1 ,108629.6,133.8,131.3,128.9
XS GIS Cut Line= 5
     1597863.421      440534.816     1597947.868      440536.516
     1598519.958      440599.799     1599145.993      440742.255
     1599655.464      441012.282
#Sta/Elev= 30
     9.4  770.57    37.5  767.83    75.1  766.37   175.3  749.04   235.9  742.35
   326.8   738.3   559.1  731.71     660  726.05   800.5  720.81   905.9     711
   920.9  710.57   935.9  711.72   981.1  714.58   991.1   716.3  1041.3  738.36
  1071.3  750.04  1081.4  752.13  1111.5  753.93  1161.6  765.21  1191.7  774.73
  1251.9  797.91    1272  803.79  1312.2  812.69  1413.4  846.99  1524.6  877.97
    1727  971.98  1797.8 1007.64  1807.9 1010.38  1828.1 1012.72  1878.7 1012.75
#Mann= 3 , 0 , 0
       0     .06       0   905.9    .045       0   935.9     .06       0
Bank Sta=905.9,935.9
XS Rating Curve= 0 ,0
Exp/Cntr=0.3,0.1

Type RM Length L Ch R = 1 ,108498.2,519.2,520.8,522.4
XS GIS Cut Line= 4
     1597940.767      440603.955     1598598.243       440751.33
      1598917.89       440800.09     1599571.854      441151.534
#Sta/Elev= 30
    10.1  781.65    30.2   781.9    80.5  773.57   150.8   766.1     171  765.49
   211.2  767.81   261.5  766.29   301.7  767.52   331.9  771.58   382.1  783.06
   412.3  782.12   432.4  776.72   522.9  736.74   563.2   725.9   714.2   720.3
   850.8  712.89   865.8  710.54   880.8  711.64   906.2   721.9   956.7   751.3
   976.9  759.84  1037.3  775.49  1097.5  796.22    1268  846.35  1378.4  870.28
  1418.5  881.35  1619.2   976.1  1629.2  978.04  1649.3  977.65  1739.6   968.1
#Mann= 3 , 0 , 0
       0     .06       0   850.8    .045       0   880.8     .06       0
Bank Sta=850.8,880.8
XS Rating Curve= 0 ,0
Exp/Cntr=0.3,0.1

Type RM Length L Ch R = 1 ,107977.5,610.8,607.7,604.6
XS GIS Cut Line= 4
     1597659.254      441106.869     1598345.688       441168.13
     1598970.123      441369.097     1599526.599      441395.986
#Sta/Elev= 30
    10.1  1000.5    40.5 1002.14    60.8  997.46    81.1  988.44   182.4   934.7
   263.5   899.1   324.3  875.56   344.6  869.83   415.5  855.72   557.4  815.01
   608.1  793.32   749.7  726.92   769.9  718.99   896.2   709.3   911.2  708.38
   926.2  709.36   991.9  715.79    1002  719.64  1062.6  757.59  1133.2  796.86
  1244.2  827.36  1284.6  844.49  1304.8  849.82  1375.5  856.42  1436.3  858.08
  1466.7  857.76  1608.5  849.51  1669.3  848.39  1790.8  849.35  1902.3  854.92
#Mann= 3 , 0 , 0
       0     .06       0   896.2    .045       0   926.2     .06       0
Bank Sta=896.2,926.2
XS Rating Curve= 0 ,0
Exp/Cntr=0.3,0.1

Type RM Length L Ch R = 1 ,107369.8,453.2,453.5,453.8
XS GIS Cut Line= 3
     1597647.235      441772.321     1598546.915      441798.408
     1599513.253        441800.8
#Sta/Elev= 30
    10.1  970.41    80.9  953.33   121.4  949.43   131.5  946.44   161.8   928.1
   171.9  924.01   232.6  904.13   303.4   877.4   394.4  871.31   596.7  826.94
     627   814.7   697.8   781.5   758.5  760.25     809  725.51   829.3   713.7
   839.4  711.57   930.3  711.54   975.7  708.77   990.7  707.66  1005.7  708.98
  1101.4  721.74  1212.1  725.92  1312.8  738.24  1373.2   748.1  1544.3  783.76
    1655  798.18  1685.2  799.43  1765.7  795.27    1806  799.23  1866.4  810.81
#Mann= 3 , 0 , 0
       0     .06       0   975.7    .045       0  1005.7     .06       0
Bank Sta=975.7,1005.7
XS Rating Curve= 0 ,0
Exp/Cntr=0.3,0.1

Type RM Length L Ch R = 1 ,106916.3,200,198.5,197
XS GIS Cut Line= 4
     1597656.656      442137.081     1598245.204      442216.032
     1599106.494      442244.742     1599530.169      442165.957
#Sta/Elev= 30
    10.1  850.43    40.3  842.96    60.4  839.91   171.1  829.15   201.3  824.84
   301.9     817   332.1  813.48   442.8  791.54   523.4  780.46     604  767.02
   685.1  749.76     756  733.09   806.7  724.16   837.1  713.99   847.3  712.17
   903.2  706.71   918.3  705.35   933.2  705.74  1070.3  712.44  1080.5  714.53
  1202.1  780.48  1222.4  790.74  1232.5  794.69  1435.3  853.61  1525.7  877.26
  1575.8  892.56    1636  906.02    1666  911.05  1796.3  927.93  1886.5  935.68
#Mann= 3 , 0 , 0
       0     .06       0   903.2    .045       0   933.2     .06       0
Bank Sta=903.2,933.2
XS Rating Curve= 0 ,0
Exp/Cntr=0.3,0.1

Type RM Length L Ch R = 1 ,106717.8,291.4,294.9,298.4
XS GIS Cut Line= 4
     1597724.104      442369.319     1598473.627      442427.572
     1598761.009      442388.737     1599498.882      442384.853
#Sta/Elev= 30
    10.2  749.36    81.3   749.1   121.9  747.71   162.5  743.81   233.7  734.29
   325.1  728.09   457.2   724.2   548.6  719.43   721.3  716.15   831.8  707.53
   906.8   704.6   921.8  704.03   936.8  704.58   981.8  711.61   991.8  715.97
  1041.8  745.16    1062   750.8  1072.1  755.91  1102.4  777.12  1112.5  782.93
  1132.7  790.41    1153  795.26  1173.2  799.16  1223.7  805.66  1304.6  813.91
    1345  819.22    1436  834.99  1476.4  839.04    1628  860.95  1779.7  886.85
#Mann= 3 , 0 , 0
       0     .06       0   906.8    .045       0   936.8     .06       0
Bank Sta=906.8,936.8
XS Rating Curve= 0 ,0
Exp/Cntr=0.3,0.1

Type RM Length L Ch R = 1 ,106422.9,770.9,770.8,771
XS GIS Cut Line= 4
     1597716.449      442629.213     1598429.046      442618.601
     1599067.836      442769.326     1599489.995      443137.992
#Sta/Elev= 30
      10  785.65    40.2  793.15    80.3  797.61   110.4  797.96   150.6  794.17
   180.7  793.79   351.3  808.47   431.6  806.06     532  795.04   592.2  784.33
   622.3  773.99   722.8  729.28     743  721.87   763.2  716.87   980.4  702.72
   995.4     702  1010.4  704.06    1056  727.57  1066.1  731.34  1096.4  733.25
  1207.4  751.02  1298.3  774.05    1369  787.64    1409   799.4  1519.1  822.39
  1559.2  836.31  1609.2  856.87  1669.3  873.63  1809.4  925.07  1929.5  966.43
#Mann= 3 , 0 , 0
      10     .06       0   980.4    .045       0  1010.4     .06       0
#XS Ineff= 2 , 0
          936.07  736.03
Permanent Ineff=
       F       F
Bank Sta=980.4,1010.4
XS Rating Curve= 0 ,0
Exp/Cntr=0.3,0.1

Type RM Length L Ch R = 1 ,105652.1,659.4,657.6,655.5
XS GIS Cut Line= 3
     1597537.249      443185.187     1598419.315      443390.856
     1599321.586      443624.712
#Sta/Elev= 30
    10.1  946.93   110.7  976.56   130.8  981.26   191.2  985.25   201.3  982.72
   231.5  960.87   281.8  936.44   332.1  917.04   452.9  877.41   543.4  840.87
   764.8  738.26   825.2  708.32   845.3  704.59   890.7  702.11   905.7   701.6
   920.7  702.45  1017.2  711.95  1047.6  718.75  1118.5  746.79  1240.1   800.3
  1260.3   805.7    1311  810.21  1361.6  823.57  1473.1  868.49  1493.3  874.43
  1533.9  882.84  1655.4  932.91  1787.2   984.1  1807.4  990.93  1837.8  997.03
#Mann= 3 , 0 , 0
       0     .06       0   890.7    .045       0   920.7     .06       0
Bank Sta=890.7,920.7
XS Rating Curve= 0 ,0
Exp/Cntr=0.3,0.1

Type RM Length L Ch R = 1 ,104994.5,205.3,205.1,204.9
XS GIS Cut Line= 4
     1597432.838      444012.057     1598190.129      444027.591
     1598628.969      444047.009     1599176.548      444074.193
#Sta/Elev= 30
    10.1  830.31   161.6   815.6   222.2  807.61     303  787.72   373.7  772.98
   414.1  766.64   454.5  761.83   474.7  758.14   575.7  732.77   585.8  732.14
   626.2  737.01   636.3  736.48     707  721.94   757.4  718.77   797.4  710.69
   872.2  698.99   887.2  698.45   902.2  698.93   967.1  702.11   987.1  706.11
    1047  728.08  1086.9  739.97  1196.7  784.38  1237.3   799.6  1470.8  865.66
  1602.8  895.85  1643.4  910.48  1694.2  931.31  1714.5  937.92    1745  946.06
#Mann= 3 , 0 , 0
       0     .06       0   872.2    .045       0   902.2     .06       0
Bank Sta=872.2,902.2
XS Rating Curve= 0 ,0
Exp/Cntr=0.3,0.1

Type RM Length L Ch R = 1 ,104789.4,818.6,826,833.5
XS GIS Cut Line= 3
     1597378.852      444197.832     1597917.158      444226.542
     1599180.383      444262.429
#Sta/Elev= 30
      10  796.32    29.9  791.42    39.9  790.44    59.9  790.34   119.8  793.75
   199.7  786.87   329.4  797.27   379.3  796.88   469.2  800.16   509.1  798.26
   589.6  788.86   690.7  768.64   741.3  755.06   908.2  703.02  923.21  698.34
   938.2  699.64   963.7  701.03  1014.2  700.73  1044.6   704.3  1074.9  713.58
  1145.7  739.03  1317.5  790.51  1368.1  801.03  1438.9     818  1519.7  841.36
  1560.2   851.4  1651.2  863.67  1701.7  872.04  1772.5  888.66  1802.8   897.6
#Mann= 3 , 0 , 0
      10     .06       0   908.2    .045       0   938.2     .06       0
Bank Sta=908.2,938.2
XS Rating Curve= 0 ,0
Exp/Cntr=0.3,0.1

Type RM Length L Ch R = 1 ,103963.4,319.8,325.7,331.7
XS GIS Cut Line= 4
     1597380.316      444541.619     1598230.849      444850.143
      1598618.43      445230.546     1598927.331      445709.522
#Sta/Elev= 30
    10.1  925.86     191  954.53   231.2  957.99   271.4  956.45   291.5  950.89
     372  914.52   492.6  872.02   633.3  816.48   693.7  796.89   743.9  784.79
   844.4  744.75   924.9  724.18   975.2  708.87  1005.3  704.76  1095.8  698.79
    1111  696.34    1126   694.9    1141  699.22  1206.5  729.51  1266.8  762.39
    1307  781.26  1397.5  813.33  1527.8   854.7  1557.8  868.38  1617.8  899.43
  1747.8   955.4  1807.8   973.5  1827.8  977.29  1917.8  982.44  2017.8  984.68
#Mann= 3 , 0 , 0
       0     .06       0    1111    .045       0    1141     .06       0
Bank Sta=1111,1141
XS Rating Curve= 0 ,0
Exp/Cntr=0.3,0.1

Type RM Length L Ch R = 1 ,103637.7,219,211.4,203.7
XS GIS Cut Line= 4
     1597394.003      444633.423     1598096.924      445087.798
     1598139.643      445293.625     1598803.728      445713.048
#Sta/Elev= 30
    10.1  959.63    70.6  974.15    90.8   977.3     121  971.09   141.2  964.12
   191.6  939.46   292.4  894.37   403.4  862.65     474  839.34   534.5  815.58
   615.1  778.32   705.9  746.03   776.5  717.82   826.9  702.43     857  700.65
   902.1  694.48   917.1  692.67   932.1  693.68  1087.5  727.69  1147.9  737.38
  1188.2  741.63    1309  784.95  1349.3   795.3  1409.7  806.49  1550.7  849.39
  1570.8   858.1  1661.5  909.25    1732  944.87  1782.3   965.2  1832.7  977.39
#Mann= 3 , 0 , 0
       0     .06       0   902.1    .045       0   932.1     .06       0
Bank Sta=902.1,932.1
XS Rating Curve= 0 ,0
Exp/Cntr=0.3,0.1

Type RM Length L Ch R = 1 ,103426.3,189.3,186,182.6
XS GIS Cut Line= 4
     1597320.216      444765.464     1597860.028      445208.187
     1598069.739      445355.762     1598815.379      445782.951
#Sta/Elev= 30
    10.1  994.49    80.9  974.45   101.2  966.85   212.5  898.78   222.6  893.79
   414.8  848.57   445.2  839.63   536.3  805.61   576.7  788.88   617.2  770.58
   737.6  711.65   781.8  693.93   796.8  690.77   811.8  691.66   905.3     702
   934.8  707.94  1015.2  729.17  1136.6  745.26  1166.9  755.04  1237.7  783.84
  1278.1  798.22  1298.3  801.62    1359  805.04  1379.2  809.36  1520.7  853.48
  1591.5  888.05  1662.3  914.45  1712.8  936.68  1763.4  951.57  1813.9  962.89
#Mann= 3 , 0 , 0
       0     .06       0   781.8    .045       0   811.8     .06       0
Bank Sta=781.8,811.8
XS Rating Curve= 0 ,0
Exp/Cntr=0.3,0.1

Type RM Length L Ch R = 1 ,103240.3,335.7,333.6,331.5
XS GIS Cut Line= 4
     1596988.945      445254.996     1597635.124      445366.917
     1598187.785       445524.82     1598815.629      445891.025
#Sta/Elev= 30
    10.1 1014.13    40.4 1011.65   121.1  991.25   161.4  973.36   272.4  916.52
   302.7   903.9   393.5  871.59   514.6  847.85   615.4  816.57   686.1  787.18
     797     733   857.5     707   882.8  692.54   887.7  690.18   897.8  689.24
   912.8  690.53  1028.9  702.22  1099.5  723.82  1230.6  754.05    1382   801.1
  1412.3  805.41  1472.9   807.1  1503.1  812.16  1573.8   838.5    1705  876.27
  1755.5  893.56  1826.2   921.2  1896.8  954.57    1917  962.54  1957.4  974.46
#Mann= 3 , 0 , 0
       0      .1       0   882.8    .045       0   912.8     .06       0
Bank Sta=882.8,912.8
XS Rating Curve= 0 ,0
Exp/Cntr=0.3,0.1

Type RM Length L Ch R = 1 ,102906.7,404.9,411.8,418.7
XS GIS Cut Line= 4
     1596959.596      445345.488     1597685.366      445732.965
     1598417.462      445797.562     1599400.768      446271.271
#Sta/Elev= 30
    10.2  990.48    91.4  987.65   121.9  982.86   172.7  962.63   274.2  910.37
   314.9  893.45   375.8  873.09   416.4  866.76   548.5  831.88   893.2  702.63
   913.3  699.37   993.9  695.98  1039.3  689.57  1054.3  688.58  1069.3  690.78
  1134.8  711.61  1245.6  741.78  1497.3  824.32  1668.8  861.72  1769.9  901.16
  1810.3  912.43  1961.9  935.51    2063  945.08  2153.9  949.02  2234.8  946.68
  2315.6  950.13  2386.4  961.86  2548.1 1003.41  2598.6 1007.18  2649.1 1002.71
#Mann= 3 , 0 , 0
       0      .1       0  1039.3    .045       0  1069.3     .06       0
Bank Sta=1039.3,1069.3
XS Rating Curve= 0 ,0
Exp/Cntr=0.3,0.1

Type RM Length L Ch R = 1 ,102495  ,309.5,313.8,318.1
XS GIS Cut Line= 4
     1596988.391      445425.102     1597634.358      445934.698
     1598050.649      446322.279     1598632.019      447520.907
#Sta/Elev= 30
    10.2  964.18   121.9  960.35     325  879.87   375.8  872.42   548.5  833.04
   619.6   814.1   802.5  748.92   843.1  744.66   924.3   724.5  1005.6  712.61
  1056.4  695.64  1092.2  690.56 1106.84  688.41  1122.2  691.03  1147.8  694.64
  1502.6   699.7  1522.8  703.62  1664.1  750.92  1714.5  762.96  1906.3  786.07
  2007.2  805.35  2108.1  810.07  2168.7  817.67    2209  818.63  2279.7  852.55
  2370.5  879.29  2481.5  927.47    2532  939.64  2562.3  939.79  2723.7  910.72
#Mann= 3 , 0 , 0
    10.2      .1       0  1092.2    .045       0  1122.2     .06       0
#XS Ineff= 2 , 0
                         1181.81          709.66
Permanent Ineff=
       F       F
Bank Sta=1092.2,1122.2
XS Rating Curve= 0 ,0
Exp/Cntr=0.3,0.1

Type RM Length L Ch R = 1 ,102181.1,781.6,778.9,776.2
XS GIS Cut Line= 4
     1596804.933      445476.402     1597477.221      446020.062
     1597671.011      446486.594      1597728.43      447182.803
#Sta/Elev= 30
    10.1  886.24   130.7  894.78   351.9  899.05   392.1  898.11   432.3  892.61
   452.4   888.7   492.6  878.61   633.4  850.15   713.8  827.18   804.3  791.88
   844.5  775.17   864.6   766.1   965.6  714.47  1006.1  696.58  1016.2  693.79
  1056.6  691.87  1157.6   691.5    1183  688.95    1198  687.29  1208.1  687.82
    1213  689.34  1218.2  690.94  1258.6  710.28  1349.6  751.21  1734.3  897.43
    1795  918.31  1835.5  930.98  1936.7  959.97  1997.5  978.92  2068.4  997.13
#Mann= 3 , 0 , 0
    10.1      .1       0    1183    .045       0    1213     .06       0
#XS Ineff= 2 , 0
          1150.7  714.92
Permanent Ineff=
       F       F
Bank Sta=1183,1213
XS Rating Curve= 0 ,0
Exp/Cntr=0.3,0.1

Type RM Length L Ch R = 1 ,101402.2,500.6,498.3,496.1
XS GIS Cut Line= 4
     1596515.448      445704.256      1596702.06      446206.674
     1597039.399      446644.497     1597426.979      447362.238
#Sta/Elev= 30
    10.1   836.8    60.7  834.87   121.3  827.97   384.3  781.97   444.9  772.76
     536   761.2   596.3   748.4   726.9  698.01     747  692.13   782.2  685.48
   797.2  684.51   812.2  687.08   827.4  689.87   917.8  694.97   978.1  701.68
   998.2  710.78  1028.4  728.86  1038.4  731.49  1078.6  735.12  1088.7  738.45
  1128.9  761.09    1139  765.17  1290.1  807.89  1330.4   820.5  1380.7  832.08
    1713  939.37  1823.8  973.63  1843.9  977.87    1854  978.42  1904.4  973.53
#Mann= 3 , 0 , 0
       0     .06       0   782.2    .045       0   812.2     .06       0
Bank Sta=782.2,812.2
XS Rating Curve= 0 ,0
Exp/Cntr=0.3,0.1
