HEC-RAS study BEECHFK.prj: BEECHFK

--- BEECHFK.g01 (geometry) --- (continued)

Type RM Length L Ch R = 1 ,100903.9,517.1,519.4,521.6
XS GIS Cut Line= 4
     1596109.738      445887.047     1596386.854      446622.738
     1596845.609      446989.013     1597376.737      447907.722
#Sta/Elev= 30
    10.1  977.95    80.6  972.44   151.2  976.98   181.4  974.51   201.6  970.15
   231.8  959.99   302.4  917.72   342.7  900.85   453.5  869.14   564.4   849.8
   715.6  801.66   786.2  777.74   998.7  686.88  1135.5  685.41  1150.5   684.4
  1165.5  687.47  1180.9  692.85  1211.2  699.61    1272   731.4  1322.6  746.39
  1443.9  807.03  1565.2  850.69  1605.6  862.43  1625.9  865.68  1979.6  864.44
  2090.8  858.73  2181.7  843.02  2252.5  834.09  2353.5  830.93  2434.4  837.61
#Mann= 3 , 0 , 0
       0     .06       0  1135.5    .045       0  1165.5     .06       0
Bank Sta=1135.5,1165.5
XS Rating Curve= 0 ,0
Exp/Cntr=0.3,0.1

Type RM Length L Ch R = 1 ,100384.5,534.8,549.4,566.4
XS GIS Cut Line= 4
     1596020.548       445926.83     1596142.222       446967.48
      1596479.56       447383.77     1596734.452       447848.12
#Sta/Elev= 30
    10.1 1010.42    40.3 1012.24     141 1007.82   171.3 1004.64   201.5  998.35
   221.6  991.87   292.2  960.03   322.4  948.42   352.6  941.62     403  934.44
   433.2  926.23   453.3   917.2   493.6  895.17   513.8   887.7   584.3  867.91
   685.1  848.57   987.3  761.07  1047.7  742.37  1088.2  737.34  1098.3  734.72
  1158.9  707.77  1224.8  683.13  1239.8  681.21  1254.8  681.81  1462.2  693.01
  1753.5   704.1  1933.4  725.72  2033.3   735.8  2063.3  736.78  2113.3  733.34
#Mann= 3 , 0 , 0
       0     .06       0  1224.8    .045       0  1254.8     .06       0
Bank Sta=1224.8,1254.8
XS Rating Curve= 0 ,0
Exp/Cntr=0.3,0.1

Type RM Length L Ch R = 1 ,99835.2 ,539.6,535,530.3
XS GIS Cut Line= 4
     1595965.029      445921.312     1596096.957      446998.549
     1595749.375      447240.703     1595583.092      448008.486
#Sta/Elev= 30
    10.1  1017.3      71 1013.82   131.9  1003.6   202.9  985.12   273.9  969.63
   334.7  952.51     426  929.88   446.3  923.07   507.1  893.18   537.6  880.72
   588.3   866.6     639  856.57   659.3  850.93   983.9  752.63    1166  690.47
  1186.1  686.72  1276.9   684.3  1302.3  681.52  1317.3   679.1  1332.3  679.89
  1387.9  690.21  1539.1  775.01  1559.3  784.28  1579.4  789.32  1599.5  789.91
  1730.5  783.63  1831.2   782.8  1911.8  784.23    2083  775.08  2294.5  788.44
#Mann= 3 , 0 , 0
       0     .06       0  1302.3    .045       0  1332.3     .06       0
Bank Sta=1302.3,1332.3
XS Rating Curve= 0 ,0
Exp/Cntr=0.3,0.1

Type RM Length L Ch R = 1 ,99300.2 ,653.4,646.3,639.2
XS GIS Cut Line= 4
     1595595.013      445860.865     1595661.335        446579.9
      1595453.19       446967.48     1595383.532      447990.908
#Sta/Elev= 30
      10  955.89    70.2  958.48   140.4   953.5   160.5  949.28   441.3  849.98
   551.6  808.98   631.8  789.08   712.1  761.93   752.1  742.59   812.1  707.91
   852.1   686.7   867.1  680.26   882.1  677.78   897.1  678.34     982  683.82
    1082  686.76    1152  691.05  1253.4  691.56  1365.2   697.8  1426.1  705.39
  1537.8  724.58  1700.3  749.11  1801.9  758.91  1842.5  758.37  1923.8  753.88
  1954.2  754.44  1974.5  757.36  2055.8  776.99  2157.3  786.61  2187.8   791.8
#Mann= 3 , 0 , 0
       0     .06       0   867.1    .045       0   897.1     .06       0
Bank Sta=867.1,897.1
XS Rating Curve= 0 ,0
Exp/Cntr=0.3,0.1

Type RM Length L Ch R = 1 ,98653.9 ,531.4,528.9,526.3
XS GIS Cut Line= 3
     1594767.359      445830.296     1594950.698      446635.966
     1595240.313      447989.754
#Sta/Elev= 30
    10.1  935.59    30.2  930.15    70.5   924.2   100.8     917   191.5   887.4
   272.1  872.18   322.4  858.22   352.7  847.47   503.8  783.79   594.5  750.43
   725.5  697.86     786  687.87   821.4  677.78   836.4  674.54   851.4  676.15
   876.8  678.98   957.6  682.55   977.8  684.76    1089  701.76  1129.4   712.6
  1149.6  715.51  1341.6  785.39  1402.3  805.65  1553.8  847.29  1584.2  854.31
    1665  860.59  1806.5  861.96  2079.3   859.7  2170.3  856.02  2210.7   856.8
#Mann= 3 , 0 , 0
       0     .06       0   821.4    .045       0   851.4     .06       0
Bank Sta=821.4,851.4
XS Rating Curve= 0 ,0
Exp/Cntr=0.3,0.1

Type RM Length L Ch R = 1 ,98125   ,1221.1,1216.9,1212.8
XS GIS Cut Line= 4
     1594412.465      445991.352     1594383.755      446680.384
     1594613.433      447139.738     1595096.711      448066.315
#Sta/Elev= 30
    10.1  921.59   172.4  898.65   243.4  883.59   375.2  862.61   395.5  857.39
   476.7  830.12   638.9   744.7   669.3  730.68   750.1   703.3   845.8   676.7
  860.95  674.21   875.8  675.83   901.1     678   971.6   675.9   991.7  679.01
  1092.4  711.19  1122.6  716.55  1193.1  749.41  1213.3   754.4  1304.7  765.97
  1406.1  767.98  1527.9  786.07  1568.5  796.38  1639.5  820.35  1771.4  858.88
  1913.4  892.16  1984.4   906.9  2014.9  909.04  2106.2  902.19  2248.2  898.32
#Mann= 3 , 0 , 0
    10.1     .06       0   845.8    .045       0   875.8     .06       0
Bank Sta=845.8,875.8
XS Rating Curve= 0 ,0
Exp/Cntr=0.3,0.1

Type RM Length L Ch R = 1 ,96908.1 ,582.7,591.3,599.9
XS GIS Cut Line= 4
     1593859.804      447046.432     1594218.675      447448.367
     1594484.239      447670.867     1594556.013      448402.963
#Sta/Elev= 30
      10  707.52    49.9  715.63    79.8  719.15   129.7   727.8   159.7  729.39
   189.6  724.54   279.4   705.5   329.3  697.93   389.2  692.53   488.9  690.27
   568.5  681.47   741.6  670.26   756.6  669.53   771.6  670.44   796.2  676.73
   835.8  692.93   855.6  695.77   875.4  703.06   915.5  724.57  1026.4  788.39
  1076.7  815.88  1117.1  833.31  1187.6  857.18  1207.7  861.75  1268.2  867.45
  1318.6  877.61  1489.9   906.2  1530.2  908.12  1600.7  915.87  1620.9   916.5
#Mann= 3 , 0 , 0
       0     .06       0   741.6    .045       0   771.6     .06       0
Bank Sta=741.6,771.6
XS Rating Curve= 0 ,0
Exp/Cntr=0.3,0.1

Type RM Length L Ch R = 1 ,96316.8 ,276.9,275.4,273.8
XS GIS Cut Line= 3
     1594111.014      446321.513     1593795.207      447060.787
     1593853.947      448476.101
#Sta/Elev= 30
      10   803.1    90.4  786.52   160.8  776.22   221.1     771   291.4  768.61
   462.2   753.1   482.3  749.54   572.8   726.8     623  715.49   733.6  695.05
   763.7  691.51   834.3  687.34   955.7   686.8  1117.6  683.35    1315  668.71
    1330  668.41    1345   668.8  1370.5  669.95  1380.6  671.72  1421.1  689.33
  1461.6  699.83  1663.9  788.72  1714.5  807.49  1734.8  810.76  1785.4   809.4
  1835.9   812.3  1896.7  820.49  1957.4  826.75  2068.7   849.5  2220.4   886.4
#Mann= 3 , 0 , 0
       0     .06       0    1315    .045       0    1345     .06       0
Bank Sta=1315,1345
XS Rating Curve= 0 ,0
Exp/Cntr=0.3,0.1

Type RM Length L Ch R = 1 ,96041.4 ,951.1,945.4,939.7
XS GIS Cut Line= 4
     1593125.719      446687.589     1593498.812       447371.32
     1593572.599      447744.139     1593742.365       448511.85
#Sta/Elev= 30
    10.1  861.92   161.8  851.28   333.8  842.88   343.9  840.09   364.2  831.51
   485.5  771.38     526  752.78   586.7   728.3   637.3  710.78   818.9  676.99
   868.9  675.65   973.9  667.01   988.9  666.53  1003.9  667.13  1028.9  672.26
  1068.9  673.82  1118.9  681.38  1179.1  698.33  1209.4  703.44  1249.7  719.02
  1269.8  723.71  1320.2  728.29  1471.4  735.15  1491.6  737.31  1511.8  745.15
    1663  820.98  1703.3  836.42  1773.8  848.91  1884.7  859.39  1945.2  872.17
#Mann= 3 , 0 , 0
       0     .06       0   973.9    .045       0  1003.9     .06       0
Bank Sta=973.9,1003.9
XS Rating Curve= 0 ,0
Exp/Cntr=0.3,0.1

Type RM Length L Ch R = 1 ,95096.1 ,347.7,349.8,352
XS GIS Cut Line= 3
     1592230.531      447419.657     1592859.841      448080.427
     1593472.224      448718.769
#Sta/Elev= 30
    10.1   841.4    30.4   836.6    50.7  833.02    81.1   830.5   131.8  828.71
   152.1  826.74   375.1   795.6   476.5  758.53   557.6  731.55   740.1  676.79
   760.4   674.3   897.5  664.54   912.5  664.19   927.5  666.24   942.7  668.77
   952.7  669.17  1033.1  668.77  1043.2  669.88  1053.2  672.38  1073.3  678.33
  1113.5  692.05  1133.6  695.06  1153.7  700.64  1284.4  750.35  1364.8  778.32
  1515.6  838.54    1596  861.71  1726.7  892.23  1756.9  898.05  1797.1  902.37
#Mann= 3 , 0 , 0
       0     .06       0   897.5    .045       0   927.5     .06       0
Bank Sta=897.5,927.5
XS Rating Curve= 0 ,0
Exp/Cntr=0.3,0.1

Type RM Length L Ch R = 1 ,94746.3 ,170.6,168.6,166.7
XS GIS Cut Line= 4
     1592035.806      447699.332      1592465.79      448078.124
     1592698.802      448458.711      1593162.66       448732.88
#Sta/Elev= 30
    10.1  812.17   211.1  759.61   311.7   738.3   341.8  728.96   412.2  702.46
   432.3  697.68   542.9  687.81   735.3  668.14   831.9     664   846.9  662.93
   861.9  664.07   867.2  665.05   907.7  686.37     928  695.58   948.3  699.41
   958.4   702.9  1019.3  733.34  1029.3  736.28  1079.2  740.96  1089.1  744.48
  1109.1  755.78    1129  765.12  1288.7   828.7  1308.7  835.39  1348.6  845.25
  1368.5  847.03  1378.5  846.21  1438.4  836.43  1478.3  832.39  1558.1  831.14
#Mann= 3 , 0 , 0
       0     .06       0   831.9    .045       0   861.9     .06       0
Bank Sta=831.9,861.9
XS Rating Curve= 0 ,0
Exp/Cntr=0.3,0.1

Type RM Length L Ch R = 1 ,94577.6 ,520.6,511.3,502.1
XS GIS Cut Line= 4
     1591991.998      447814.043      1592333.75       448260.65
     1592605.597      448555.799     1593028.903      448843.181
#Sta/Elev= 30
      10  853.44    70.3  844.17   170.7  815.87   180.8  811.66   210.9  795.91
     241  783.19   391.6  725.53     482  693.85   552.3  688.76   572.4  684.45
   612.5  672.26   622.6  670.71     758  663.17     773  662.31     788  662.85
   813.2  669.16   873.3  694.75   903.4  700.06   913.5  703.33   993.7  735.36
  1003.8   738.4  1033.9  742.89  1043.9  746.63  1164.3  804.88  1214.4  827.82
  1224.5  829.99  1234.5  829.55    1395  795.73  1435.1     785  1475.3  770.92
#Mann= 3 , 0 , 0
      10     .06       0     758    .045       0     788     .06       0
#XS Ineff= 2 , 0
          729.26  686.77
Permanent Ineff=
       F       F
Bank Sta=758,788
XS Rating Curve= 0 ,0
Exp/Cntr=0.3,0.1

Type RM Length L Ch R = 1 ,94066.3 ,436.6,440.6,444.6
XS GIS Cut Line= 4
     1591433.838      448747.479     1592086.983      448919.737
     1592689.886      448862.318     1593356.784      449042.026
#Sta/Elev= 30
    10.1  826.15    40.3  816.01     121  794.93   302.5  755.83   403.3  745.27
   584.7  718.16   625.1  715.05   715.9  688.15   796.6  673.96   857.2  665.66
     933  662.48     948  661.91     963  662.78  1018.7  666.37  1079.2  691.76
  1109.5  697.19  1170.1   720.1  1291.3  749.86  1331.9   752.8  1443.6  753.14
  1545.2  740.34  1585.8  729.31    1596  729.26  1616.3  738.14    1728  813.27
  1799.1  847.34  1819.4   853.6  1860.1  861.38  1951.5  872.67  1971.8  873.55
#Mann= 3 , 0 , 0
    10.1     .06       0     933    .045       0     963     .06       0
#XS Ineff= 2 , 0
          888.19  684.67
Permanent Ineff=
       F       F
Bank Sta=933,963
XS Rating Curve= 0 ,0
Exp/Cntr=0.3,0.1

Type RM Length L Ch R = 1 ,93625.7 ,416.2,419.5,422.5
XS GIS Cut Line= 4
     1591476.903       448912.56     1592180.289      449206.834
     1592653.999      449350.382     1593142.063      449450.866
#Sta/Elev= 30
      10  855.55   100.3  838.95   180.6  829.13   361.2  820.98   421.4  816.27
   451.5  805.65   561.8   757.6   642.1  729.18   722.3  694.81   752.4  684.62
   792.8  683.98     813   681.6   863.5  665.43   873.6  663.93    1015  664.48
  1040.4  661.11  1055.4   659.1  1070.4  662.81  1085.7  666.98  1126.1  670.91
  1186.7  684.39  1347.1  763.92  1367.1  771.45    1387  771.68  1426.9  765.64
  1626.2  732.58  1695.9  718.56  1705.9  719.08  1725.8  724.37  1755.7   738.5
#Mann= 3 , 0 , 0
       0     .06       0  1040.4    .045       0  1070.4     .06       0
Bank Sta=1040.4,1070.4
XS Rating Curve= 0 ,0
Exp/Cntr=0.3,0.1

Type RM Length L Ch R = 1 ,93206.2 ,621,622.3,623.9
XS GIS Cut Line= 3
      1591428.86      449024.691     1592175.143      449578.587
     1592947.364      450084.937
#Sta/Elev= 30
    10.1  894.48    80.8  890.01   151.5  889.62   232.3  891.32   303.1  880.59
   353.6   869.4     394  858.16   434.4  844.65   545.5  800.84     596  783.28
   636.4  763.37   656.6  755.31   717.2   736.1   747.5  725.14   818.3  695.67
   858.7  680.31   924.5  660.46   939.5  659.02   954.5  661.25   980.1  663.39
  1122.2  666.48  1152.6  673.11  1172.9  676.08  1203.4   691.7  1304.8   736.6
  1355.6  756.67  1477.3  801.14  1548.4  830.91  1761.5   883.2  1852.8  907.15
#Mann= 3 , 0 , 0
       0     .06       0   924.5    .045       0   954.5     .06       0
Bank Sta=924.5,954.5
XS Rating Curve= 0 ,0
Exp/Cntr=0.3,0.1

Type RM Length L Ch R = 1 ,92583.9 ,320.3,316.5,312.8
XS GIS Cut Line= 4
      1591299.08      449199.178     1591627.628      449824.091
     1592072.628      450269.091     1592575.066      450564.101
#Sta/Elev= 30
    10.1  934.87    50.4  929.95    90.8  921.87   242.1  881.95   363.1  847.86
   393.4  835.92     585  750.27   726.3  693.58   766.9  681.88   817.7  679.51
   827.8  677.81   858.3  666.93     894  657.79     909   654.7     924  655.63
   949.6  659.37  1051.1  659.35  1122.2  661.55  1142.5  664.84  1162.8  672.43
  1193.2  678.21  1203.4  682.22  1335.3  742.22  1385.6  762.12  1465.9  787.57
  1616.6  832.33  1717.1  838.93  1817.5  850.47  1867.8  850.71    1918  847.39
#Mann= 3 , 0 , 0
       0     .06       0     894    .045       0     924     .06       0
Bank Sta=894,924
XS Rating Curve= 0 ,0
Exp/Cntr=0.3,0.1

Type RM Length L Ch R = 1 ,92267.3 ,474.6,480.6,486.6
XS GIS Cut Line= 4
     1590048.597      450111.188     1591283.113      450111.188
     1591986.499      450333.688      1592516.54      450643.327
#Sta/Elev= 30
    10.1  790.87    60.7  784.58   273.2  750.21   354.2  732.34     425  714.68
   475.6  700.69   526.2  681.98   546.4  678.41   586.9  677.77   647.6     670
   799.4  665.38  1032.1  665.99  1153.6  662.68  1598.3  658.12  1618.5     657
  1633.9   653.5  1648.9   651.6  1663.9  653.93  1689.3  657.78    1760   659.8
  1820.7  673.74  1901.5  714.14  2012.5  760.16  2082.9  786.49    2244  834.01
  2314.4  838.13  2354.7   837.5  2394.9  834.44  2525.7  818.84  2586.1  814.35
#Mann= 3 , 0 , 0
    10.1     .06       0  1633.9    .045       0  1663.9     .06       0
#XS Ineff= 2 , 0
          1361.6  675.85
Permanent Ineff=
       F       F
Bank Sta=1633.9,1663.9
XS Rating Curve= 0 ,0
Exp/Cntr=0.3,0.1

Type RM Length L Ch R = 1 ,91786.7 ,305,298.7,292.4
XS GIS Cut Line= 4
     1590285.452      450261.913     1591147.887      450258.356
     1591505.612      450721.268      1592300.23      451018.741
#Sta/Elev= 30
    10.1   806.6   152.2  781.67   233.4  763.92   365.3  714.87     487  681.72
   507.3  678.05   547.9  676.93   608.8  667.89   912.9  667.77   963.3  661.65
  1104.5  657.77  1225.6  657.99  1250.9  654.59  1265.9  651.21  1280.9  653.56
  1306.3  660.62  1326.4     663  1376.9  694.96  1447.5  722.45  1508.1  753.95
  1518.2  757.51  1528.3  757.93  1639.4  712.51  1780.8  677.95  1821.2  663.15
    1902  664.59  2033.3   673.4  2174.7  675.41  2225.2  670.92  2295.9  675.84
#Mann= 3 , 0 , 0
       0     .06       0  1250.9    .045       0  1280.9     .06       0
Bank Sta=1250.9,1280.9
XS Rating Curve= 0 ,0
Exp/Cntr=0.3,0.1

Type RM Length L Ch R = 1 ,91488   ,260.1,257.5,254.8
XS GIS Cut Line= 5
     1590341.493        450580.8     1590912.374      450724.491
     1591425.001      450868.182     1591793.397      450850.573
     1592261.893      451063.526
#Sta/Elev= 30
    10.1  832.42    50.7  826.78    81.2  818.56   121.8  799.62   192.8  775.62
   253.7  771.32   324.8  753.64   416.1  726.53   558.2  675.14   608.8  670.55
     649  660.47   869.9  657.66   925.3  651.41   940.3  651.01   955.3  651.81
  1050.8  665.76  1170.9  724.49  1190.8  729.97  1290.5  702.17  1380.2  681.26
  1430.1  675.22  1489.9  674.09  1540.3  662.06  1661.4  666.21  1711.9  670.64
  1812.8  668.66  1853.2  671.68  1913.7  670.96  1974.2  684.52  2004.5  685.43
#Mann= 3 , 0 , 0
       0     .06       0   925.3    .045       0   955.3     .06       0
Bank Sta=925.3,955.3
XS Rating Curve= 0 ,0
Exp/Cntr=0.3,0.1

Type RM Length L Ch R = 1 ,91230.5 ,931.6,934.4,937.8
XS GIS Cut Line= 4
     1590363.576      450745.922     1590887.218      451058.116
      1591547.54      451079.648     1592240.526      451284.028
#Sta/Elev= 30
       0  780.26    10.2  780.26    91.4  747.78   142.3  733.02   172.7  717.58
   193.1  711.52   243.9  721.17   365.8  726.92   436.9  717.05   518.2  691.02
   558.8  680.79   679.7  662.22   709.7  659.79     930  656.58   957.5  651.75
  970.06  650.72   982.5  652.21  1040.1  663.21  1080.1  666.34  1130.2  658.24
  1160.2  656.56  1320.5  663.65  1380.7  669.98  1410.8  677.19  1571.4  725.75
  1691.8  767.54  1792.1  784.08  1812.2  784.73  1962.7  774.31  1992.8  774.89
#Mann= 3 , 0 , 0
       0     .06       0   957.5    .045       0   982.5     .06       0
#XS Ineff= 2 , 0
                         1086.29          719.12
Permanent Ineff=
       F       F
Bank Sta=957.5,982.5
XS Rating Curve= 0 ,0
Exp/Cntr=0.3,0.1

Type RM Length L Ch R = 1 ,90296.1 ,534.3,541.9,549.3
XS GIS Cut Line= 3
     1590306.984      451690.219     1591361.892      451865.337
     1592201.822      452027.557
#Sta/Elev= 30
    10.1  810.36    70.6  811.69     111  809.12   262.3   790.7   312.7  786.57
   373.3  777.57   423.7  764.93   474.1  746.93   534.7  727.32   665.8  699.26
     686  694.02   756.6  661.45   766.7  657.23   776.8   654.9   938.2  657.28
  1039.1  654.77  1054.3  652.49 1069.67  650.09  1084.3  652.21  1099.5  657.65
  1139.8  678.59    1170  685.54  1320.9  762.11  1381.3  791.65  1431.7  815.33
  1451.8  821.56  1763.8  895.98  1773.8  895.54  1783.9  893.45  1924.8  858.31
#Mann= 3 , 0 , 0
    10.1     .06       0  1054.3    .045       0  1084.3     .06       0
Bank Sta=1054.3,1084.3
XS Rating Curve= 0 ,0
Exp/Cntr=0.3,0.1

Type RM Length L Ch R = 1 ,89754.1 ,365.2,357.1,349
XS GIS Cut Line= 4
     1589976.823      451927.074     1590795.048      451948.606
     1591189.806       452465.38      1592044.08      452555.819
#Sta/Elev= 30
    10.1  703.59   161.7   704.6   363.8  723.15   565.9  724.34   636.6  722.04
   818.5  708.09   930.3  692.58  1001.4  671.66  1031.9  655.81    1042  654.23
  1199.8  651.22  1214.8  649.04  1229.8  651.36  1265.6  656.99  1296.1  672.34
  1316.4  676.33    1357  693.91  1367.2  695.71  1468.8  692.31  1519.3  709.08
    1580  733.54    1681  790.22  1731.6  811.95  1792.2  826.82    2055  882.48
  2115.6  906.35  2186.4  940.95  2206.6   944.2  2267.2  947.47  2327.9  944.08
#Mann= 3 , 0 , 0
    10.1     .06       0  1199.8    .045       0  1229.8     .06       0
Bank Sta=1199.8,1229.8
XS Rating Curve= 0 ,0
Exp/Cntr=0.3,0.1

Type RM Length L Ch R = 1 ,89397   ,702.6,701,701.4
XS GIS Cut Line= 4
     1590003.625       452318.95     1590449.325      452514.135
     1591292.506      452611.229     1592046.368      452660.702
#Sta/Elev= 30
    10.1  709.91    30.4  700.02    50.7  694.05   121.6  681.05   182.5  675.05
   243.3   671.9   324.4   665.3   486.6  658.67   865.6  648.16   880.6  646.66
   895.6   648.4  920.99  654.98  1082.7   651.6    1204  658.55  1254.5  666.92
  1274.7  675.35  1335.3  705.52  1405.8  743.36  1456.2  773.38  1486.4  787.82
  1597.2  819.26  1728.2  843.62  1768.5  853.31  1828.9  872.94    1849  880.75
  1939.7  925.73  2010.2  945.79  2030.4  950.12  2050.5  952.05  2090.8  948.02
#Mann= 3 , 0 , 0
    10.1     .06       0   865.6    .045       0   895.6     .06       0
#XS Ineff= 2 , 0
          688.45  821.25
Permanent Ineff=
       F       F
Bank Sta=865.6,895.6
XS Rating Curve= 0 ,0
Exp/Cntr=0.3,0.1

Type RM Length L Ch R = 1 ,88696.1 ,917.2,924.1,929
XS GIS Cut Line= 3
     1590030.444      453026.252     1591220.967      452988.218
     1592069.318      453128.281
#Sta/Elev= 30
    10.1  672.31    50.5   673.3   141.3  690.95   282.6  684.94   343.2  685.93
   625.8  719.84   676.3   722.7   726.8  730.46     747  728.67   767.2  722.93
     858   681.5   928.7  656.91     959  653.68  1150.8  652.28  1176.1  648.15
  1191.1  645.71  1206.1  650.83  1221.5  659.11  1241.7  663.52  1251.8  669.85
  1302.4  711.64  1342.9  734.44  1383.3  752.62  1454.1  779.05  1595.8  823.88
  1656.5  835.97  1858.8  886.07  1899.2  900.77    1970  932.52    2051   950.1
#Mann= 3 , 0 , 0
       0     .06       0  1176.1    .045       0  1206.1     .06       0
Bank Sta=1176.1,1206.1
XS Rating Curve= 0 ,0
Exp/Cntr=0.3,0.1

Type RM Length L Ch R = 1 ,87772   ,267.4,265,262.6
XS GIS Cut Line= 4
      1589596.42      453262.073     1590393.113      453470.218
     1590889.072      453852.949     1591853.891      453854.451
#Sta/Elev= 30
      10  687.48    30.1  683.44   140.6  680.92   210.9  703.44   301.3  739.94
   451.9  783.65     482  787.17   572.4  760.91   662.8  719.19   733.1  700.94
   823.4  686.42   914.4   660.7  1025.5  650.92  1237.7  650.82  1263.1  647.38
  1278.1  645.21  1293.1  648.72  1328.6   656.1  1429.7  721.51  1500.7  759.85
  1541.3  776.47  1754.6  810.02  1866.3  832.46  1998.3  833.28  2028.8  830.77
  2191.3     776  2282.7  758.98  2313.2   748.8  2333.5  749.44  2414.7  780.19
#Mann= 3 , 0 , 0
       0     .06       0  1263.1    .045       0  1293.1     .06       0
Bank Sta=1263.1,1293.1
XS Rating Curve= 0 ,0
Exp/Cntr=0.3,0.1

Type RM Length L Ch R = 1 ,87507   ,415.5,402,388.5
XS GIS Cut Line= 4
      1589657.99      453495.663      1590316.46      453812.124
     1590691.012      453981.106     1591832.773      453946.154
#Sta/Elev= 30
    10.1  753.47   202.9  803.41   213.1  805.41   223.2  804.39     345  744.74
   537.8   684.3   629.1  659.21   669.7  656.36   880.9  652.26   976.1  646.16
   991.1  644.62  1006.1  647.41  1061.3  656.08  1131.5  659.75  1181.9  666.35
  1353.8  724.26  1384.1  738.06  1454.8  775.37  1525.6  801.84  1646.9  828.51
    1748  844.22  1778.3  846.17  1798.5  844.12    1930  815.16  2051.3   766.3
  2111.9   743.9  2132.1  734.27  2142.2  732.37    2213  745.55  2283.8  763.71
#Mann= 3 , 0 , 0
    10.1     .06       0   976.1    .045       0  1006.1     .06       0
Bank Sta=976.1,1006.1
XS Rating Curve= 0 ,0
Exp/Cntr=0.3,0.1

Type RM Length L Ch R = 1 ,87105   ,711.6,714.2,716.9
XS GIS Cut Line= 4
     1589755.872      454376.995     1590529.484      454467.878
        1590874.      454022.879     1591830.874       454010.17
#Sta/Elev= 30
    10.1   898.4   131.5  853.82   252.9  818.56   374.3   777.1   455.2  752.94
   627.2  728.09     698  725.53   758.7  717.19   849.3   687.7   929.7  647.63
  1080.4   647.4  1105.6  644.81  1120.6  643.01  1135.6  645.24    1191  652.17
  1241.2  668.84  1281.4  677.48  1392.1  718.99  1452.5  748.97  1573.4  803.55
    1654   819.8  1754.7  833.92  1815.2  835.14  1946.1   808.4  2097.2  746.36
  2157.6  734.01  2187.9  721.38  2197.9  723.66  2218.1  733.71  2298.7  751.74
#Mann= 3 , 0 , 0
       0     .06       0  1105.6    .045       0  1135.6     .06       0
Bank Sta=1105.6,1135.6
XS Rating Curve= 0 ,0
Exp/Cntr=0.3,0.1

Type RM Length L Ch R = 1 ,86390.7 ,460.2,461.1,462.6
XS GIS Cut Line= 3
     1589799.628      454537.906     1590988.839      454876.991
     1591814.241      454238.201
#Sta/Elev= 30
    10.1  899.11   111.5  884.14     223  852.81   253.4  847.17   314.2   841.1
   425.7  836.55   496.7  829.24   527.1  824.18   729.8  775.87   851.4  737.34
   881.8  730.67  1135.2  692.03  1236.6  682.89  1348.1  652.74  1449.4  648.67
  1474.9  642.77  1489.9  641.21  1504.9  644.04  1560.9  649.28  1621.7  673.12
  1652.1   676.4  1733.1  692.13  1834.5  708.72  1925.7  711.56  2006.7  707.73
  2128.3  692.02  2168.9     679    2179  678.21  2209.4  681.38  2280.3  698.85
#Mann= 3 , 0 , 0
       0     .06       0  1474.9    .045       0  1504.9     .06       0
Bank Sta=1474.9,1504.9
XS Rating Curve= 0 ,0
Exp/Cntr=0.3,0.1

Type RM Length L Ch R = 1 ,85929.6 ,700.5,711.1,721.7
XS GIS Cut Line= 4
     1589861.951      454652.647     1591265.169      455168.573
     1591878.838      454833.926     1593463.252      455500.529
#Sta/Elev= 30
    10.1  904.41   171.7  888.26   282.8  857.56   555.6  799.39   767.7  786.01
   979.9  765.92  1151.6  738.61  1242.5  712.42  1495.1  667.22  1576.1  675.75
  1596.4  670.08  1652.3   642.6 1667.02  641.17  1682.3  644.48  2062.3  655.17
  2153.5  674.04  2183.9  689.45  2355.8  727.92    2467  738.88  2497.4  738.89
  2537.8  731.36  2729.9  675.52  2901.8  682.68  3043.4  715.98  3306.3  792.15
  3599.5  865.78  3660.2  884.63  3801.7  898.08  3892.8  914.43    3913  913.93
#Mann= 3 , 0 , 0
    10.1     .06       0  1652.3    .045       0  1682.3     .06       0
Bank Sta=1652.3,1682.3
XS Rating Curve= 0 ,0
Exp/Cntr=0.3,0.1

Type RM Length L Ch R = 1 ,85218.5 ,974.8,985.2,995.7
XS GIS Cut Line= 4
     1590018.093      454809.703     1591148.536      455186.517
     1592350.753      455958.089     1592745.511       456927.04
#Sta/Elev= 30
    10.1  858.26    80.8  837.01   363.5  779.64   403.9  775.64   626.1   768.3
   727.1   757.2   858.3  732.84   959.3  718.22  1070.4   689.7  1292.9  646.89
  1677.9  647.67  1880.5  646.03  1895.9  642.96 1910.52  640.74  1925.9  644.02
  2012.2  672.99  2184.5  695.22  2356.7  747.14  2447.9  767.34  2528.9  791.74
  2549.2   803.7    2610  872.75  2630.3  890.88  2681.1  908.89  2721.7  917.96
  2823.3  923.19  2985.8  922.75  3229.6  961.32  3442.9   947.1  3666.4  906.76
#Mann= 3 , 0 , 0
    10.1     .06       0  1895.9    .045       0  1925.9     .06       0
Bank Sta=1895.9,1925.9
XS Rating Curve= 0 ,0
Exp/Cntr=0.3,0.1

Type RM Length L Ch R = 1 ,84233.3 ,1106.1,1093.1,1081.4
XS GIS Cut Line= 4
     1589698.755      454745.154     1590897.326      455186.517
     1590834.524      455868.371     1591641.983      457061.616
#Sta/Elev= 30
    10.1  918.95   243.3  879.63   415.6  820.54   658.9   773.3   881.9  749.47
  1277.3  690.29  1413.3  641.04  1428.3  639.64  1443.3  642.23  1508.9   646.5
  1780.7  646.98  1831.1   666.1  1881.4  695.11  1911.6  702.78  2012.7  744.27
  2043.2   750.9  2235.9  750.64  2286.7  738.19  2337.4   701.3  2347.6   699.9
  2418.6  730.65  2591.1  782.55  2641.8  806.46  2682.4  817.98    2794  863.82
    2865  881.31  2946.2  895.98  3078.1  900.68    3281   943.3  3402.8  918.86
#Mann= 3 , 0 , 0
       0     .08       0  1413.3    .045       0  1443.3     .06       0
Bank Sta=1413.3,1443.3
XS Rating Curve= 0 ,0
Exp/Cntr=0.3,0.1

Type RM Length L Ch R = 1 ,83140.2 ,348,350.2,351.1
XS GIS Cut Line= 4
     1589306.897      455658.249     1589820.714      455563.331
     1590655.089      455778.653     1591516.378       457079.56
#Sta/Elev= 30
      10  868.62   190.9  794.24   401.9  718.57   603.6  664.75   694.9  654.24
     984  638.25     999  638.15    1014   639.1  1130.8  648.29  1272.7  692.43
  1343.7  696.64  1384.2  703.27  1455.1  735.06  1495.7  747.13  1515.9  749.41
  1627.4  739.03  1698.3   741.4  1738.8  736.32  1840.1  713.94  1890.8  694.54
    1911  692.48    1982  724.32  2113.7  766.28  2366.9  864.62  2488.5   892.5
  2691.1  916.65    2762  930.39  2802.6   933.6  2853.2  929.32  2944.4  907.09
#Mann= 3 , 0 , 0
       0     .08       0     984    .045       0    1014     .06       0
Bank Sta=984,1014
XS Rating Curve= 0 ,0
Exp/Cntr=0.3,0.1

Type RM Length L Ch R = 1 ,82790   ,409.4,407,404.6
XS GIS Cut Line= 4
     1589281.287       455740.35      1589964.79      455868.507
     1590423.048      456109.286     1591157.037      456854.926
#Sta/Elev= 30
    10.1  890.81    50.4  879.72    80.6  867.62   201.6  804.45     262  778.09
   312.4  758.71   403.1  729.89   483.8  709.26   665.2  653.01   685.3  649.89
   715.7  648.59   979.6  642.52  1005.2  639.77 1020.19  638.06  1035.2  638.65
  1121.7  649.36  1233.4  651.31  1263.9  653.01  1395.9  668.06  1436.6  683.72
  1538.1  712.08  1649.9   729.5    1721  747.47  1842.9   792.3  1974.9  835.32
    2046  860.71    2107  875.63  2157.8  886.18  2228.9  898.31  2259.4  901.11
#Mann= 3 , 0 , 0
    10.1     .08       0  1005.2    .045       0  1035.2     .06       0
Bank Sta=1005.2,1035.2
XS Rating Curve= 0 ,0
Exp/Cntr=0.3,0.1

Type RM Length L Ch R = 1 ,82383   ,1026.2,1030.6,1035
XS GIS Cut Line= 4
     1589181.669      455879.018     1589722.025      456191.355
     1590520.512      456424.621     1590757.852      456891.613
#Sta/Elev= 30
    10.1  902.69    50.3  897.66   110.7   884.1   140.9  873.87   231.5  837.18
     302  817.38   392.6  789.16   463.1   775.3   483.2  769.57   513.4   758.9
   614.1  717.57     685  693.53   806.7  656.95   837.2  642.88   847.3   640.4
   903.3  638.52  917.77  637.84   933.3  638.37   979.2  641.24  1161.8  644.97
  1344.4   662.1    1456   693.8  1566.8  732.72  1717.9  765.42  1768.3  781.05
  1848.9  810.28  1899.2  826.17  1949.6  838.62  1969.8  840.43  1979.8  839.15
#Mann= 3 , 0 , 0
    10.1     .08       0   903.3    .045       0   933.3     .06       0
Bank Sta=903.3,933.3
XS Rating Curve= 0 ,0
Exp/Cntr=0.3,0.1

Type RM Length L Ch R = 1 ,81352.4 ,515.3,514,512.6
XS GIS Cut Line= 4
     1589004.448      456143.402     1589282.408      456819.379
     1589973.234      457330.769     1590343.934      457509.749
#Sta/Elev= 30
    10.2  827.34   101.5  787.18   142.1  773.12   213.2  753.63   314.7  728.53
     467   694.9   527.9  677.51   588.8  656.18   619.2  656.61   730.9  671.26
   801.7  655.04   882.6  648.42     908  641.57   923.2  637.74     938  639.48
   963.5  642.45  1115.1  643.27  1256.7  646.93  1297.2  658.99  1317.4  662.36
  1347.7  678.39  1357.8  682.26  1479.2  722.74  1590.4  753.55  1620.5  759.85
  1680.8  761.22  1791.2  757.85  1821.3  759.04  1871.5  764.02  2002.1  770.87
#Mann= 3 , 0 , 0
    10.2     .08       0     908    .045       0     938     .06       0
Bank Sta=908,938
XS Rating Curve= 0 ,0
Exp/Cntr=0.3,0.1

Type RM Length L Ch R = 1 ,80838.4 ,157.6,156.2,154.8
XS GIS Cut Line= 3
      1588125.05      456693.774     1589704.081      457590.951
     1590231.135      457758.971
#Sta/Elev= 30
    10.1  920.65   131.9   921.5   243.5  914.97   294.2  914.82   365.3  906.24
   456.6  882.04     558  871.61   608.8  862.23   659.5  845.52   771.1  796.84
     903  746.59  1085.6   660.8  1136.3  640.08  1329.1   642.4    1446  639.47
 1471.15  637.11    1476  638.53  1491.4   641.7    1532  662.73  1562.5  673.03
  1592.9  689.63  1633.5  704.24  1856.3  759.33  1997.2  784.86  2047.4   814.1
  2067.6  823.17  2117.9  832.34  2218.4  859.03    2309  870.43  2369.3  872.38
#Mann= 3 , 0 , 0
    10.1     .08       0    1446    .045       0    1476     .06       0
Bank Sta=1446,1476
XS Rating Curve= 0 ,0
Exp/Cntr=0.3,0.1

Type RM Length L Ch R = 1 ,80682.2 ,311.8,310,308.2
XS GIS Cut Line= 4
     1588046.321      457181.143      1588912.35      457336.485
      1589603.62      457654.935     1589991.975       457736.49
#Sta/Elev= 30
    10.1  866.97    50.6  865.13   212.4  836.72   293.3  828.57   333.7  818.37
   485.4  794.01   586.6  771.51   647.2  764.63   768.6  741.49   829.3  732.29
   859.6  723.83   900.1  707.81   930.6  691.02  1001.6  646.71  1021.9  638.81
  1214.7  641.96  1260.6  638.44 1275.61  636.43  1290.6   638.2  1356.8  644.62
  1377.1  651.32  1407.5  666.43  1448.1  674.39  1650.9  736.37  1769.9  764.91
  1839.4  774.92    1879  784.44  1928.6  801.83  1978.2  826.09  2037.8  841.33
#Mann= 3 , 0 , 0
    10.1     .08       0  1260.6    .045       0  1290.6     .06       0
Bank Sta=1260.6,1290.6
XS Rating Curve= 0 ,0
Exp/Cntr=0.3,0.1

Type RM Length L Ch R = 1 ,80372.1 ,1418.5,1411.1,1403.3
XS GIS Cut Line= 4
     1587828.982      458075.426     1588796.648      457723.716
     1589498.765      457821.928     1590045.008      457797.301
#Sta/Elev= 30
    10.1  770.58    90.8  763.73   121.1  759.28   191.8  743.39   343.2  715.91
     434  693.46   464.3  687.73   585.5  670.05   706.6  655.27   827.7  649.03
  1394.2  639.71  1429.8  637.02  1444.8  635.87  1459.8  637.06  1495.5  640.49
  1505.6   643.7  1546.1  675.92  1556.3  680.49  1576.5  684.03    1617  701.09
  1647.4  706.88    1698  713.57  1758.8  725.83  1910.7  751.13  2001.8  768.76
  2022.1  775.11  2113.2  814.85  2163.8  834.07  2224.6  849.14  2285.4  859.65
#Mann= 3 , 0 , 0
    10.1     .06       0  1429.8    .045       0  1459.8     .06       0
#XS Ineff= 2 , 0
         1116.33  661.15
Permanent Ineff=
       F       F
Bank Sta=1429.8,1459.8
XS Rating Curve= 0 ,0
Exp/Cntr=0.3,0.1

Type RM Length L Ch R = 1 ,78961   ,268.2,270.9,274
XS GIS Cut Line= 3
     1588860.735      459376.332     1589641.525      458942.752
     1590281.217      458544.453
#Sta/Elev= 30
    10.1  820.66    40.6  826.34    60.9  827.11      71  826.06   162.4  804.58
   294.3  776.73   334.9  766.78   456.7  731.45   507.4  715.29   558.2   696.1
     680  645.95   690.1  642.24   700.3     640   801.8  639.82   878.1  634.88
   893.1  634.78   908.1  634.85   993.6  635.59  1013.7  636.94  1023.7  639.03
  1053.9  651.92    1094  660.54  1124.2   665.6  1174.4  685.28  1214.6  698.59
    1295  714.85  1345.2  722.07    1516  737.89  1616.5  744.82  1646.7  745.08
#Mann= 3 , 0 , 0
       0     .06       0   878.1    .045       0   908.1     .06       0
Bank Sta=878.1,908.1
XS Rating Curve= 0 ,0
Exp/Cntr=0.3,0.1

Type RM Length L Ch R = 1 ,78690.1 ,390.4,394.1,398.4
XS GIS Cut Line= 4
     1588854.097      459433.597     1589498.765       459239.42
     1590007.509      459099.612     1590357.027      459095.729
#Sta/Elev= 30
      10   799.9    30.1  806.42    60.3  812.83    80.4   814.9   100.5  814.88
   120.6  813.01   150.7  806.84   281.4  787.17   341.7   772.7   422.1  755.21
   482.3  738.18   552.7  715.43   683.4  667.67   754.4  643.83   774.7  639.15
   784.9  637.92   825.5  635.17   861.2     634   876.2  633.88   891.2  634.23
  1129.9  644.08  1170.4  646.94  1190.7  654.67  1250.8  684.84  1270.8  693.58
  1340.7  715.52  1390.6  729.36  1410.6  734.32  1430.6  737.86  1550.4     750
#Mann= 3 , 0 , 0
       0     .06       0   861.2    .045       0   891.2     .06       0
Bank Sta=861.2,891.2
XS Rating Curve= 0 ,0
Exp/Cntr=0.3,0.1

Type RM Length L Ch R = 1 ,78296.1 ,721.4,727.4,732.7
XS GIS Cut Line= 3
     1588753.074      459519.881     1589727.739      459571.779
     1590466.682      459645.485
#Sta/Elev= 30
    10.1  741.85    50.3   753.3   120.7  765.75   181.1  772.05   281.7  777.51
   372.3  776.04   462.9  766.91   553.4  761.34   593.7  755.29   654.1  741.97
   724.5  733.09   764.7  721.79   794.9  707.53     815  693.68   875.4  647.22
   895.5  637.84   935.8  633.68   991.2  633.32  1006.2  633.28  1021.2  633.31
  1166.7  636.75  1216.9  648.66  1297.2  692.51  1447.7  741.41    1538  772.95
  1568.1  789.87  1628.3     836  1648.4  848.75  1678.5  861.63  1718.7  871.54
#Mann= 3 , 0 , 0
       0     .06       0   991.2    .045       0  1021.2     .06       0
Bank Sta=991.2,1021.2
XS Rating Curve= 0 ,0
Exp/Cntr=0.3,0.1

Type RM Length L Ch R = 1 ,77568.7 ,495.8,493.2,491.2
XS GIS Cut Line= 4
     1588657.059      459568.758     1589218.659      459928.824
     1589621.583      460206.042     1590294.207       460758.05
#Sta/Elev= 30
    10.1  689.18   101.1  696.05   212.3   695.6   323.4  703.55   363.9  702.89
   505.4   692.9   586.3  685.14   866.7  642.81   896.7  642.85   966.5  635.47
  1126.2  635.78  1161.4  633.43  1176.4  633.07  1191.4  633.43  1257.4   637.9
  1297.8  648.68  1328.2  653.47  1388.9  678.89  1429.4  698.27  1449.6  709.91
    1480  730.75  1500.2  741.21  1672.2  810.07  1702.6  825.04  1722.8  831.41
  1803.7  841.96  1844.2  841.62  1884.7  833.95  1935.3  819.06  2026.3   798.1
#Mann= 3 , 0 , 0
       0     .06       0  1161.4    .045       0  1191.4     .06       0
Bank Sta=1161.4,1191.4
XS Rating Curve= 0 ,0
Exp/Cntr=0.3,0.1

Type RM Length L Ch R = 1 ,77075.5 ,630,625.2,619.7
XS GIS Cut Line= 4
      1588407.49      460000.594     1588896.816      460350.113
       1589537.6      460711.282     1590112.364      460913.226
#Sta/Elev= 30
      10   748.2    60.1  751.89    90.2  750.16   110.2   746.9   180.4  729.73
   270.6  700.38   481.1  647.83   521.2  646.83     692  637.69  1024.5  635.98
  1059.9  633.12  1074.9  631.96  1089.9   632.5  1155.5  635.14  1185.8  639.64
    1216  651.55  1236.1  654.45  1246.2  657.68  1266.4  666.99  1296.6  683.81
    1347  702.33  1377.5  715.43  1397.8  720.55  1438.4  721.83  1468.9   720.1
  1509.5  715.36  1550.1  713.82  1651.7  714.61  1763.3  723.56  1946.1  732.77
#Mann= 3 , 0 , 0
       0     .06       0  1059.9    .045       0  1089.9     .06       0
Bank Sta=1059.9,1089.9
XS Rating Curve= 0 ,0
Exp/Cntr=0.3,0.1

Type RM Length L Ch R = 1 ,76450.3 ,797.9,802.9,807.8
XS GIS Cut Line= 4
     1588187.853      460300.425     1588618.497      460686.211
     1589594.017      460782.028     1590124.464      460991.048
#Sta/Elev= 30
    10.1  847.61    50.7  825.01   162.3  794.21   233.3  783.96   294.2  780.48
   395.6  760.37   476.7  731.26   507.2  723.83   537.6  712.66   578.2     705
   638.8  681.39   739.9  658.03   800.5  637.26     836  628.82     851  626.97
     866  629.18   891.4  633.08  1063.2  633.08  1305.8  637.96  1346.2  652.15
  1376.5  659.37    1427  677.56  1487.7   688.2  1558.4  704.95  1598.4  704.82
  1758.4  696.17  1918.5   700.6  1958.5  707.14  2028.5  730.36  2128.5  749.51
#Mann= 3 , 0 , 0
       0     .06       0     836    .045       0     866     .06       0
Bank Sta=836,866
XS Rating Curve= 0 ,0
Exp/Cntr=0.3,0.1

Type RM Length L Ch R = 1 ,75647.4 ,602.8,608.7,614.6
XS GIS Cut Line= 4
     1588080.191      460551.634     1588815.876      461116.855
     1589479.787      461520.585     1590125.754      461475.726
#Sta/Elev= 30
    10.1   827.8    60.5  823.71   110.9  825.49   231.9  852.93   272.3  853.08
   292.4  848.24   312.6  839.33   373.1  825.51   433.6  804.11   524.4  782.39
   685.7  760.82     716  752.83   857.2  727.53   877.3  721.11  1089.2  634.66
  1149.8  631.74  1391.9  631.78  1427.4  627.74  1442.4  625.72  1457.4  627.29
  1533.2  648.08  1704.8  706.74  1735.1  711.03  1795.8  731.69  1866.7  749.36
  1947.6  774.17  2079.1  789.46  2220.8  815.46  2311.8  821.91  2352.3  831.29
#Mann= 3 , 0 , 0
       0     .06       0  1427.4    .045       0  1457.4     .06       0
Bank Sta=1427.4,1457.4
XS Rating Curve= 0 ,0
Exp/Cntr=0.3,0.1

Type RM Length L Ch R = 1 ,75038.8 ,770.2,759.4,748.5
XS GIS Cut Line= 4
     1587416.281      460847.702     1588501.864      461224.517
     1588824.848      461771.794      1589919.21      461880.744
#Sta/Elev= 30
    10.1  871.72    40.3  873.94    60.5  869.71   211.7  814.79   393.1   764.6
   453.6  735.39   564.5  741.16   715.7  701.97   735.8   700.2   806.4  724.34
   846.7  733.27   977.8  744.37  1108.8  743.05  1149.1  733.61  1330.7   635.5
    1467  629.49 1482.03  625.54    1497  626.88  1532.4  632.46  1613.1  636.74
  1633.3  647.06  1784.6  701.37  1925.9   734.1  2097.4  757.89  2198.3  754.21
  2258.8  757.83  2410.2  780.68  2531.2  806.75  2682.6  815.86  2884.4  842.63
#Mann= 3 , 0 , 0
    10.1     .06       0    1467    .045       0    1497     .06       0
Bank Sta=1467,1497
XS Rating Curve= 0 ,0
Exp/Cntr=0.3,0.1

Type RM Length L Ch R = 1 ,74279.4 ,1197.4,1187.8,1178.3
XS GIS Cut Line= 4
     1586662.652      462211.411     1587721.321      461969.173
     1588860.553      461954.029      1589901.46      462040.947
#Sta/Elev= 30
    10.1  814.29    30.4  816.71    50.7  813.71     203  780.75   345.1  809.81
   497.3  816.34     680  833.87   751.1  844.88   842.4  846.46   893.2  852.31
  1136.4  765.79  1307.8   673.2  1378.4  643.03  1418.8  634.19  1655.8  626.95
 1670.84  625.44  1685.8  628.42    1812  636.24  1842.2  650.35  1892.6  658.53
  1993.5  690.79  2296.3  745.22  2367.3  746.17  2438.3   737.5  2590.4  736.18
  2651.3  743.35  2762.8  765.19  3016.4  819.92  3138.1  819.37  3269.9  802.92
#Mann= 3 , 0 , 0
    10.1     .06       0  1655.8    .045       0  1685.8     .06       0
Bank Sta=1655.8,1685.8
XS Rating Curve= 0 ,0
Exp/Cntr=0.3,0.1

Type RM Length L Ch R = 1 ,73091.5 ,1190.5,1195.5,1200.3
XS GIS Cut Line= 4
      1588235.05      463170.542     1588753.074      462785.604
     1589183.719      462175.524     1589659.223      462121.693
#Sta/Elev= 30
    10.1  698.82    30.3  705.17    50.4  709.62    90.8  713.82   312.6  711.62
   342.9  708.55   373.1  703.91   443.7  687.48   494.1   672.5   514.3  665.41
   544.5  652.57   554.6  651.37   645.4  643.91   857.3  632.25   968.3  629.18
  1129.8  629.29  1155.1  626.97 1169.95  625.37  1185.1  627.85  1210.5  634.55
  1230.7  637.39  1271.1  649.06  1392.1  688.46  1461.9  713.37  1491.8  722.44
  1531.7   732.5  1571.6  740.66  1671.3  757.86  1751.1  774.16  1870.7  785.01
#Mann= 3 , 0 , 0
    10.1     .06       0  1155.1    .045       0  1185.1     .06       0
Bank Sta=1155.1,1185.1
XS Rating Curve= 0 ,0
Exp/Cntr=0.3,0.1

Type RM Length L Ch R = 1 ,71896.1 ,795.6,800,805.8
XS GIS Cut Line= 3
     1588582.696      463711.564     1589450.087      463154.852
     1590204.465      462652.554
#Sta/Elev= 30
    10.1   737.2   181.9  704.28   202.1  706.44   303.1  731.26   323.3  734.73
   373.9  737.54   434.5  731.45   505.2  720.59   626.5  693.51   717.4  679.76
   757.9  667.84   848.8  636.46   858.9  634.36  1015.7  624.32  1030.7  623.42
  1045.7  625.19    1071  628.23  1272.4  630.79  1322.7  637.41  1342.8  644.81
  1443.5  690.88  1493.9   710.4  1594.6  726.05  1634.9  726.06  1665.1   723.1
  1745.7  709.08    1796  696.85  1856.4  689.22  1896.7  688.32    1937  693.09
#Mann= 3 , 0 , 0
       0     .06       0  1015.7    .045       0  1045.7     .06       0
Bank Sta=1015.7,1045.7
XS Rating Curve= 0 ,0
Exp/Cntr=0.3,0.1

Type RM Length L Ch R = 1 ,71096.1 ,664.2,666.4,676.7
XS GIS Cut Line= 3
     1588676.371      463873.065     1589899.447      463699.968
      1590751.71      463676.001
#Sta/Elev= 30
    10.1   731.4      81  716.36   192.4  687.67   212.6  684.83   263.3  695.38
   374.6  723.64   394.9  726.22   496.1  707.74   556.9  699.43   587.3  697.54
     648  697.75   678.4  693.68   739.1  675.92   820.1  644.61   860.6  631.67
  1220.3  622.63  1235.3  620.73  1250.3  622.06  1316.5  631.73  1346.9  641.45
  1377.4  646.35  1397.7  646.44  1438.3  641.44  1509.3  655.21    1621  688.48
  1773.2  743.03  1905.2  783.14  1996.5   818.4  2067.6  850.44  2087.9  856.79
#Mann= 3 , 0 , 0
       0     .06       0  1220.3    .045       0  1250.3     .06       0
Bank Sta=1220.3,1250.3
XS Rating Curve= 0 ,0
Exp/Cntr=0.3,0.1

Type RM Length L Ch R = 1 ,70429.7 ,612.3,601.4,590.5
XS GIS Cut Line= 4
     1588044.304      464292.861     1589300.352      464068.567
     1590018.093      464463.325      1590738.23      464045.833
#Sta/Elev= 30
    10.1  746.25   313.9  727.89   415.2  685.18   475.9   667.5   486.1  668.31
   607.6  707.81   668.3  714.85   779.7  718.95   860.7  727.07     962  703.82
  1053.1  668.77  1073.4  663.76  1194.9  699.21  1296.1  705.51  1366.9   683.9
  1518.6  628.81  1614.9   621.7  1629.9  620.37  1644.9  621.08  1862.5   628.1
    1913  645.29  2024.3  698.13  2044.5  701.03  2095.1  698.38  2379.3  746.41
  2551.9  785.06  2602.6  803.28  2663.5  834.03  2704.1  850.03  2927.5  905.76
#Mann= 3 , 0 , 0
       0     .06       0  1614.9    .045       0  1644.9     .06       0
Bank Sta=1614.9,1644.9
XS Rating Curve= 0 ,0
Exp/Cntr=0.3,0.1

Type RM Length L Ch R = 1 ,69828.3 ,488,481.9,475.8
XS GIS Cut Line= 5
     1588924.972      465657.456     1589279.345       464905.02
     1589924.983      464492.394     1590143.433      464472.976
     1590784.217       464147.73
#Sta/Elev= 30
    10.1  682.79    50.7  672.29    91.3  666.36   233.3  658.48   263.7  652.62
   608.6  659.21     710  653.19   730.3  647.63   760.7  635.87     781   633.2
   932.5   628.6  1335.8  626.45 1374.56  621.52  1411.5  620.62  1426.5   618.9
  1441.5   624.3 1458.97  625.81 1474.35  630.54    1477  635.89  1507.2  641.69
  1567.7  669.38  1597.9  678.86  1677.7   690.8  1817.3  700.88  1898.2  714.14
  2181.6  777.15    2212  788.42  2353.7  855.25  2485.2  896.78  2535.9  908.79
#Mann= 3 , 0 , 0
    10.1     .06       0  1411.5    .045       0  1441.5     .06       0
#XS Ineff= 2 , 0
         1343.12  628.24
Permanent Ineff=
       F       F
Bank Sta=1411.5,1441.5
XS Rating Curve= 0 ,0
Exp/Cntr=0.3,0.1

Type RM Length L Ch R = 1 ,69346.4 ,642.6,645.7,649.5
XS GIS Cut Line= 4
     1589192.691      466042.356     1589973.234      465342.558
     1590295.916       464579.53     1590856.078      464184.695
#Sta/Elev= 30
    10.1  807.09    80.6  779.18     131  770.74   332.6  762.77   473.8  744.48
   554.4  736.16   655.2  731.46     756  731.49   856.8  720.63   917.3  710.74
  1048.3  684.38  1189.8  630.31 1280.51   624.3    1503  620.81  1583.8  621.67
  1609.2  619.06  1624.2  617.24  1639.2  618.85 1675.76  629.53  1694.9  632.08
  1755.5  661.49  1785.8  673.72  1896.9   703.2  1967.5  726.19  2148.9   764.2
  2199.3  777.85  2239.6  792.55  2370.6  848.94  2501.6  886.66  2562.1  906.05
#Mann= 3 , 0 , 0
    10.1     .06       0  1609.2    .045       0  1639.2     .06       0
Bank Sta=1609.2,1639.2
XS Rating Curve= 0 ,0
Exp/Cntr=0.3,0.1

Type RM Length L Ch R = 1 ,68700.7 ,856.7,861.4,865.4
XS GIS Cut Line= 3
     1590009.121      466006.469      1590638.44       465274.11
     1591285.845      464613.891
#Sta/Elev= 30
    10.1  768.06    50.3  751.49    80.5  735.28    90.5  733.22   100.6  734.69
   130.8  745.19   201.2  758.64   251.5   769.9   261.5  769.55   452.6  718.15
   573.3  678.95   593.4  670.91   643.7  644.16   673.9  629.68     694  622.43
   875.1  619.65   925.4  620.98   950.6  618.31   965.6  617.03   980.6  619.09
  1016.4  630.25  1057.1  648.86  1128.2   670.5    1240  701.27  1372.1  731.82
  1443.2  753.04  1504.2  778.59  1646.4  848.87    1809  906.59  1890.3  932.56
#Mann= 3 , 0 , 0
       0     .06       0   950.6    .045       0   980.6     .06       0
Bank Sta=950.6,980.6
XS Rating Curve= 0 ,0
Exp/Cntr=0.3,0.1

Type RM Length L Ch R = 1 ,67839.3 ,1188.8,1197.9,1207.1
XS GIS Cut Line= 4
     1589076.058      466544.775     1590739.148      466073.656
     1591588.153      465719.372      1592054.88       465578.38
#Sta/Elev= 30
    10.1  930.38   151.6  915.34   242.6  899.55   454.9  851.64   525.6  831.73
   566.1  816.14   616.6  804.43   869.3  762.49  1051.3  726.26    1122  718.38
  1162.5  704.54  1233.2  661.32  1314.1  648.65  1415.2  646.25    1496  657.93
    1860  677.56  1920.6  671.07  2092.5   623.9  2229.1  618.74  2244.1  616.99
  2259.1  619.29    2325  631.85  2547.4  705.25  2668.8  725.09  2790.7  782.73
  2882.1  819.75  2983.7  855.03  3095.4  908.97  3115.7  911.33  3136.1  906.87
#Mann= 3 , 0 , 0
       0     .06       0  2229.1    .045       0  2259.1     .06       0
Bank Sta=2229.1,2259.1
XS Rating Curve= 0 ,0
Exp/Cntr=0.3,0.1

Type RM Length L Ch R = 1 ,66641.4 ,880.1,891,855.3
XS GIS Cut Line= 4
     1589641.279      468007.173     1590628.173      466742.154
     1591256.197       467127.94     1592151.556      466677.995
#Sta/Elev= 30
    10.2  875.33     325  809.96   416.3  804.31   538.2  780.11   670.2  781.21
   863.1  736.29  1015.5  708.56  1066.2  705.08    1249   715.1  1340.4  708.49
    1442  695.88  1543.5  676.81  1604.4  675.61  1786.2  624.72  2018.4  619.43
  2043.8  615.68  2058.8  614.84  2073.8  616.74  2139.6  640.57  2270.8  669.34
  2351.6  706.06  2432.6  731.26  2493.3  761.76  2513.6  768.03  2867.8  835.61
  3029.8  877.36  3120.9  910.55  3161.4  921.28  3292.9  936.92  3343.5  932.98
#Mann= 3 , 0 , 0
       0     .06       0  2043.8    .045       0  2073.8     .06       0
Bank Sta=2043.8,2073.8
XS Rating Curve= 0 ,0
Exp/Cntr=0.3,0.1

Type RM Length L Ch R = 1 ,65750.4 ,738.1,733.6,729
XS GIS Cut Line= 4
     1590372.971       468079.26     1590699.948      467845.681
     1591489.463      467388.121     1592172.784      466822.002
#Sta/Elev= 30
      10  812.88    90.4  811.11   160.7     806   180.8  801.89   200.9  792.65
   281.3  741.77   381.7  710.96   503.2  657.68   564.1  642.92   614.8  623.79
   624.9  622.02   883.7  616.31   898.7   614.7   913.7   615.5   989.9  637.17
  1121.7  664.46    1142  673.53  1294.1  753.98  1314.4  761.67  1475.7  790.59
  1717.7  841.34    1869  867.82  1889.1  873.28  1929.5  893.47  1979.9  915.44
  2000.1  920.66  2050.5  926.56    2111  927.14  2171.5   924.3  2201.7  917.67
#Mann= 3 , 0 , 0
       0     .06       0   883.7    .045       0   913.7     .06       0
Bank Sta=883.7,913.7
XS Rating Curve= 0 ,0
Exp/Cntr=0.3,0.1

Type RM Length L Ch R = 1 ,65016.9 ,616.2,608.4,600.5
XS GIS Cut Line= 4
     1590928.329      468603.572     1591336.943       468500.62
     1591767.588      467782.879     1591991.882      467172.799
#Sta/Elev= 30
      10  765.87   120.4  782.05   200.7  786.04   220.7  784.44   260.9  772.58
   391.3  727.67   451.6  710.25     492   691.7   572.7  650.49   592.8  642.99
   633.2  632.23   663.4  627.07   865.1  619.87   890.4  616.53   905.4  614.23
   920.4  615.62     976  624.64  1056.7  646.77  1248.3  711.22  1258.4  711.76
  1319.3  701.33  1410.8  696.13  1431.1  698.76  1461.5  705.79  1502.2  717.16
  1573.3  752.01  1603.7  763.92  1654.5  780.22  1837.3  831.03  1908.4  846.22
#Mann= 3 , 0 , 0
      10     .06       0   890.4    .045       0   920.4     .06       0
#XS Ineff= 2 , 0
          753.42  649.41
Permanent Ineff=
       F       F
Bank Sta=890.4,920.4
XS Rating Curve= 0 ,0
Exp/Cntr=0.3,0.1
